HEC-RAS study DRKFK_2.prj: DRKFK_2

--- DRKFK_2.g01 (geometry) --- (continued)

Type RM Length L Ch R = 1 ,70161   ,645,645,645
XS GIS Cut Line= 2
2378021.17796652685770.9882197332378611.36306695686400.804595268
#Sta/Elev= 30
       0 2601.09    97.1 2561.32   112.6 2553.32   123.6 2552.05   133.1 2548.65
   145.5 2547.71   162.1 2541.17   167.8 2540.12     215 2538.01   396.3 2537.28
   402.7 2535.97     414 2530.67   430.6 2527.57     564 2529.32   583.5 2530.69
   594.42525.635   603.6 2522.65   623.4 2522.25   653.7 2522.84  667.612525.635
   694.2 2530.94   706.4 2534.95   723.9 2535.99   745.1 2543.36   764.9 2553.91
   770.7 2559.29   776.2  2562.3   790.4 2565.56   801.7  2573.3   863.1 2601.77
#Mann= 6 ,-1,0
       0     .05       0     230     .07       0     410     .06       0
     550     .05       0   594.4    .045       0  667.61      .1       0
#XS Ineff= 2 , 0
          490.97 2536.57
Permanent Ineff=
       F       F
Bank Sta=594.4,667.61
XS Rating Curve= 0 ,0
Exp/Cntr=0.3,0.1

Type RM Length L Ch R = 1 ,69516   ,618.2,618.2,618.2
XS GIS Cut Line= 2
2377618.85324163686447.5732751072378333.02068412686895.116650642
#Sta/Elev= 30
       0 2585.86    29.9    2574    70.8 2553.47   133.7 2547.55   153.7 2542.89
   190.4 2530.39   204.5 2527.59   239.3 2525.64   280.1  2525.4   294.2 2522.95
   321.3 2524.65   393.4 2523.18   412.2 2524.52   431.1 2523.41  435.592521.547
   443.2 2519.01   459.5 2518.71   489.7 2518.87  506.862521.546   549.1 2523.97
   577.5 2522.86   601.1 2526.85   681.3 2526.02   695.5 2531.11   714.4 2534.16
     738 2546.11   788.6 2574.55   822.9 2587.15   837.1 2589.29   842.8 2591.45
#Mann= 5 ,-1,0
       0      .1       0     110     .05       0     220     .06       0
  435.59    .045       0  506.86      .1       0
Bank Sta=435.59,506.86
XS Rating Curve= 0 ,0
Exp/Cntr=0.3,0.1

Type RM Length L Ch R = 1 ,68897   ,542.4,542.4,542.4
XS GIS Cut Line= 2
2377345.28491845687311.4815064192378273.59557639687269.504963504
#Sta/Elev= 30
       0 2598.55    22.9 2587.99    30.9 2582.19    42.9 2579.12      71  2566.6
      95 2560.11     139 2531.78   163.1 2524.41   199.1 2523.18   215.1 2520.94
   243.1  2522.7   275.2 2519.59   531.4 2520.33   539.4 2518.94  546.072515.685
   551.5 2513.54   575.5 2513.18   607.5  2513.5  615.23 2515.72   627.5 2519.92
   671.5 2520.81   767.7 2518.95   783.7 2515.28   807.7 2516.25   815.7 2520.91
   843.9 2545.14   863.8 2559.57   879.8 2563.64   887.8 2570.15   929.3 2592.93
#Mann= 8 ,-1,0
       0      .1       0     170     .06       0     270     .05       0
     370     .06       0     460     .08       0  546.07    .045       0
  615.23     .08       0     660      .1       0
#XS Ineff= 2 , 0
          305.42 2524.85
Permanent Ineff=
       F       F
Bank Sta=546.07,615.23
XS Rating Curve= 0 ,0
Exp/Cntr=0.3,0.1

Type RM Length L Ch R = 1 ,68355   ,732,732,732
XS GIS Cut Line= 3
2377686.76786648687810.427114398 2377899.2124616687831.906646366
 2378358.4611266687757.977743771
#Sta/Elev= 30
       0 2545.88    37.6 2535.34    53.7 2532.52     126 2529.19   154.2 2521.04
   175.4 2521.16   226.7  2518.3   230.7 2516.82   236.5 2510.73   238.8 2508.58
   242.9 2508.22   271.2 2507.86   287.4 2507.98   303.1 2510.73     336 2513.04
   364.4 2511.56   380.6 2513.93   421.1 2515.35     454 2512.23   509.9 2512.79
   514.3 2514.79   522.4 2523.19   530.5 2529.25   550.8 2539.69   562.2 2550.35
   607.5 2578.34   619.7 2580.42   628.5 2587.16     648 2595.37   678.7 2611.43
#Mann= 5 ,-1,0
       0     .05       0     120     .06       0  223.53      .1       0
   236.5    .045       0   303.1      .1       0
Bank Sta=236.5,303.1
XS Rating Curve= 0 ,0
Exp/Cntr=0.3,0.1

Type RM Length L Ch R = 1 ,67623   ,454.8,454.8,454.8
XS GIS Cut Line= 2
2377453.74493531688539.1679251032378419.82126637688447.968925103
#Sta/Elev= 30
       0 2561.01     6.5 2555.81    34.6 2539.33    70.1 2526.17    86.8 2524.43
     127 2524.99   143.1 2523.45   211.4 2523.58   275.7 2521.56   359.9 2523.51
   444.4 2517.09   468.5 2519.48   476.5 2518.75   492.6 2521.52   536.8    2520
   551.1 2512.69   576.8 2511.88     589 2507.81   733.7 2509.17   773.9 2510.84
   777.9 2510.64  786.822506.167     806 2503.73   834.1 2503.25   854.2 2503.46
  861.662506.166   870.3 2515.49   894.4 2537.32   926.5 2563.88   970.4 2569.33
#Mann= 7 ,-1,0
       0      .1       0      60     .05       0     450      .1       0
     460     .06       0     550      .1       0  786.82    .045       0
  861.66      .1       0
Bank Sta=786.82,861.66
XS Rating Curve= 0 ,0
Exp/Cntr=0.3,0.1

Type RM Length L Ch R = 1 ,67168   ,509.9,509.9,509.9
XS GIS Cut Line= 3
2377851.36394211689164.3721140462377881.09943671689092.049880597
2378446.00628765688866.273548086
#Sta/Elev= 30
       0 2546.55    23.2 2543.55      64 2526.59   104.3 2522.24   167.7 2518.14
   240.9 2515.87   290.7 2509.04     323 2510.47   374.4 2507.53   402.8 2507.95
   421.8 2502.99   434.7 2501.56   443.4 2501.38   455.2 2502.69   464.9 2505.03
     495  2504.3   529.5 2507.17   533.8 2506.89  540.79 2503.29   546.7 2501.66
   589.8 2501.28   615.7 2501.57  622.17 2503.32   636.7 2515.41   654.4 2523.05
   661.4  2527.9     667  2532.9     676  2544.6   678.7 2546.68   686.6 2548.66
#Mann= 5 ,-1,0
       0     .05       0   208.2     .06       0   428.2      .1       0
  540.79    .045       0  622.17      .1       0
#XS Ineff= 2 , 0
        399.8679    2512
Permanent Ineff=
       F       F
Bank Sta=540.79,622.17
XS Rating Curve= 0 ,0
Exp/Cntr=0.3,0.1

Type RM Length L Ch R = 1 ,66658   ,582.2,582.2,582.2
XS GIS Cut Line= 3
2378103.61354591689767.0976920082378443.44324447689607.091649903
 2378727.5070102689173.156975324
#Sta/Elev= 30
       0 2550.83    13.9 2541.72    23.3 2532.71      36 2528.58    49.3 2519.88
    62.5 2513.87    75.8 2509.65   124.4 2508.23   150.9 2500.78   164.2 2498.81
   186.3 2498.58   358.7 2505.76   409.3 2504.09   435.4 2504.78   502.2 2500.01
   526.1  2501.3   565.3 2500.56     596 2497.76   640.5 2498.75   660.7 2501.82
   693.4 2497.74   748.9 2498.93   779.1 2496.75   796.42498.988   808.2 2506.85
   822.4 2521.71   836.9 2531.33     859 2540.77   880.9 2547.71   894.3 2554.88
#Mann= 7 ,-1,0
       0      .1       0     210     .05       0  415.61     .06       0
  535.61     .05       0  645.61      .1       0   748.9    .045       0
   796.4      .1       0
#XS Ineff= 2 , 0
             339    2512
Permanent Ineff=
       F       F
Bank Sta=748.9,796.4
XS Rating Curve= 0 ,0
Exp/Cntr=0.3,0.1

Type RM Length L Ch R = 1 ,66076   ,525.3,525.3,525.3
XS GIS Cut Line= 2
2378658.27151386690226.3492529422379179.82261344689553.905192518
#Sta/Elev= 30
       0 2523.56    27.8 2512.66      45 2508.86   117.9 2505.34     139 2498.62
   146.7 2497.44   230.3 2496.16   239.4 2494.75   269.8 2496.91     330 2495.64
   458.3 2497.15   497.6 2499.34   543.1 2495.74   588.7 2493.78   629.7 2495.35
   664.6 2494.74   677.9 2496.91   689.9 2500.59  701.092493.629     708 2490.99
   714.5 2490.47   760.2 2490.76  767.912493.629     776 2497.97     789 2511.21
   801.3 2520.94   812.4 2527.87   826.6 2543.56   831.8 2546.99     851  2554.6
#Mann= 6 ,-1,0
       0     .05       0     330     .06       0     570     .05       0
     700      .1       0  701.09    .045       0  767.91      .1       0
#XS Ineff= 2 , 0
           497.6    2512
Permanent Ineff=
       F       F
Bank Sta=701.09,767.91
XS Rating Curve= 0 ,0
Exp/Cntr=0.3,0.1

Type RM Length L Ch R = 1 ,65551   ,524.7,524.7,524.7
XS GIS Cut Line= 2
 2379265.4528889690314.8567144582379612.01211199689832.083868681
#Sta/Elev= 30
       0 2520.57    21.8 2517.99    54.7 2511.33      71 2510.79    75.9 2509.71
    93.8  2502.3   105.5 2500.77   149.3 2497.95   203.9 2495.82   248.3 2495.64
   258.3 2496.49   272.9 2495.72   297.5 2496.19   356.6 2495.63     370 2494.65
   400.9 2491.97   407.3 2489.58   410.8 2488.17   415.7 2487.67   484.6 2487.47
   513.4 2487.76  518.52 2489.57   524.8 2494.71   539.2 2503.21   548.6    2511
   553.5 2516.18   559.2  2524.1   563.4 2528.64   582.2 2540.15   594.3    2546
#Mann= 6 ,-1,0
       0     .05       0     180     .06       0     300     .05       0
     370      .1       0   407.3    .045       0  518.52      .1       0
Bank Sta=407.3,518.52
XS Rating Curve= 0 ,0
Exp/Cntr=0.3,0.1

Type RM Length L Ch R = 1 ,65026   ,617,617,617
XS GIS Cut Line= 2
2379760.86599461690483.7309997122380073.58750848690055.249505597
#Sta/Elev= 30
       0 2526.73      30 2523.26    44.3 2522.08    55.7 2519.84    67.2  2519.7
    72.5 2518.18    87.2 2511.21    95.8  2505.9   112.1 2492.63   115.8  2491.4
   136.9    2491   161.6 2488.47   196.3 2488.84   236.3 2487.85   317.7 2491.89
     325 2491.05  335.272483.733   350.6 2481.38   358.4 2481.09   409.2 2481.64
   413.6 2482.16   417.32483.733   424.1 2488.24   448.8 2511.08   458.7 2521.67
     468 2528.93     488 2542.38   503.3 2550.18   513.8 2554.55   530.5 2563.59
#Mann= 5 ,-1,0
       0      .1       0      30     .06       0     190      .1       0
  335.27    .045       0   417.3      .1       0
Bank Sta=335.27,417.3
XS Rating Curve= 0 ,0
Exp/Cntr=0.3,0.1

Type RM Length L Ch R = 1 ,64409   ,639.3,639.3,639.3
XS GIS Cut Line= 3
2379920.80570978690958.1280445982380050.41570613690900.973528166
2380506.21894808690544.810989798
#Sta/Elev= 30
       0 2551.91    73.6 2524.12    91.3 2518.35   104.2 2511.94   117.3 2510.13
   126.1  2506.8   141.1 2503.57   168.4 2500.51   219.3 2498.69   265.7 2491.93
   305.2 2490.35   342.2 2485.78   436.3 2486.46   459.6 2485.42   468.8 2483.14
   496.1 2485.06   507.5 2482.82   538.9 2482.02  548.062479.866   555.1 2477.52
   565.2 2476.84   605.8 2477.03  632.012479.866   636.3 2482.02   661.7  2502.5
   678.5 2513.55   692.1  2526.5   698.4 2535.84   702.3 2540.39   720.1 2551.79
#Mann= 7 ,-1,0
       0      .1       0  291.65     .07       0  371.65     .05       0
  531.65     .07       0  541.65      .1       0  548.06    .045       0
  632.01      .1       0
#XS Ineff= 2 , 0
        436.4471    2492
Permanent Ineff=
       F       F
Bank Sta=548.06,632.01
XS Rating Curve= 0 ,0
Exp/Cntr=0.3,0.1

Type RM Length L Ch R = 1 ,63770   ,373.9,373.9,373.9
XS GIS Cut Line= 3
2380073.15741447691304.752243396 2380679.8247179691217.283669285
2380764.82988818691168.884707561
#Sta/Elev= 30
       0 2532.31    23.3 2523.46    35.4 2516.65    47.5 2515.17    63.7 2507.85
      96 2499.46   116.2 2497.45   156.6 2496.39   201.1 2490.97   241.5 2487.28
   265.7 2483.66   281.9 2482.14   394.4 2480.85   403.1  2480.1   411.2 2478.33
   447.6  2480.6   451.6 2480.07  463.042475.667   468.5 2474.13   496.1 2473.81
   572.9 2473.94  577.562475.666   597.1 2492.75   608.5 2501.63   627.2 2515.56
   636.4 2520.34   651.4 2531.41   671.9 2543.25     687 2550.29   710.8 2562.91
#Mann= 6 ,-1,0
       0     .06       0     200     .05       0     370     .06       0
     400     .07       0  463.04    .045       0  577.56      .1       0
Bank Sta=463.04,577.56
XS Rating Curve= 0 ,0
Exp/Cntr=0.3,0.1

Type RM Length L Ch R = 1 ,63396   ,346.8,346.8,346.8
XS GIS Cut Line= 3
2380295.54280083691533.6052948722380727.06156355  691629.3814105
2381002.81257778691474.666146794
#Sta/Elev= 30
       0 2483.37     8.8 2481.83    86.7 2476.96   152.2 2475.72   172.7 2476.24
   180.9  2477.6   197.3 2475.02   230.1 2473.85   250.6 2475.51   275.2 2472.63
   275.2 2472.61   287.5 2469.89   303.9 2469.76   348.8 2470.02   355.6 2472.64
   365.3 2476.97     394 2477.02   418.6 2479.52   530.4 2477.16   556.9 2477.71
   567.1 2479.28   575.2 2482.83   590.1 2492.14     622 2516.31   640.5 2529.04
   695.7  2560.9   713.3 2569.49   727.7 2578.03   751.5  2593.8   758.2 2595.88
#Mann= 5 ,-1,0
       0     .06       0      70      .1       0     170     .07       0
   275.2    .045       0   355.6      .1       0
Bank Sta=275.2,355.6
XS Rating Curve= 0 ,0
Exp/Cntr(USF)=0,0
Exp/Cntr=0.3,0.1

Type RM Length L Ch R = 1 ,63049   ,272.3,272.3,272.3
XS GIS Cut Line= 4
2380374.93046111692055.007015446 2380738.5724389691828.369910817
2380921.28322128691668.355142256 2380995.0893879691607.556042857
#Sta/Elev= 30
       0 2560.53    41.3 2546.62    57.4 2543.55   128.7 2524.12   138.2 2517.49
   152.3 2493.44   161.7 2482.02   167.7 2476.41   171.1 2474.45   199.7 2472.83
   207.6 2469.04   213.6 2466.49   228.7 2466.22     256  2466.3  266.87 2469.01
   278.1 2473.02   298.4 2476.22   369.1 2474.56   391.3 2474.73   425.7 2477.42
   462.5 2475.48   511.3 2477.54   632.7 2475.64   664.6 2477.42     670 2479.13
   685.5  2487.9   711.4 2505.86   742.5 2529.68   758.1 2537.16     767 2542.99
#Mann= 6 ,-1,0
       0      .1       0   207.6    .045       0  266.87     .06       0
     340      .1       0  458.49     .05       0  588.49      .1       0
#XS Ineff= 2 , 0
                         428.899            2480
Permanent Ineff=
       F       F
Bank Sta=207.6,266.87
XS Rating Curve= 0 ,0
Exp/Cntr=0.3,0.1

Type RM Length L Ch R = 1 ,62777   ,594.3,594.3,594.3
XS GIS Cut Line= 2
2380674.48865064692228.0578142722381104.15133114 691741.92465547
#Sta/Elev= 30
       0 2509.86    28.7 2487.04    42.9 2473.29    45.7 2472.47    57.2 2472.77
    74.1 2471.48   83.58 2466.97    91.1 2464.66   110.6 2464.38   158.7 2464.66
  164.942466.968   170.4 2468.86   181.8 2469.48   195.9  2472.2   233.4 2476.36
   262.3 2477.56   318.8 2473.61     371 2473.98   395.1 2471.45   414.1 2474.04
   430.9 2475.03   484.3 2471.93   527.5 2473.09     553  2477.3   558.7 2479.03
   581.3 2494.03   606.6 2508.14   623.8 2519.08   635.2 2524.99   648.8 2530.65
#Mann= 5 ,-1,0
       0     .06       0   83.58    .045       0  164.94      .1       0
     390     .05       0     520      .1       0
#XS Ineff= 1 ,-1
 268.102 648.795    2480
Permanent Ineff=
       F
Bank Sta=83.58,164.94
XS Rating Curve= 0 ,0
Exp/Cntr=0.3,0.1

Type RM Length L Ch R = 1 ,62183   ,412.4,412.4,412.4
XS GIS Cut Line= 2
2381125.95448253692660.6360719612381498.64921618692059.965667959
#Sta/Elev= 30
       0 2542.06      39 2518.27    51.1  2515.2    72.5 2503.43    79.7 2497.24
   102.8 2471.44   105.8  2469.4   146.5 2467.39   152.3  2465.6  157.56 2462.07
   164.1 2459.93   192.4 2459.64   234.7 2459.85  244.12 2462.05   253.6 2465.36
   269.8 2468.55   385.4 2471.19     437 2467.81   492.2 2468.28   527.7 2471.84
   542.9 2477.09   564.2 2486.99   599.6 2505.37   611.3 2508.44   625.4 2515.73
   634.9 2517.52   658.4 2529.49   671.9 2532.06   681.9 2537.79   706.9 2545.66
#Mann= 6 ,-1,0
       0      .1       0      50     .06       0  157.56    .045       0
  244.12      .1       0     390     .05       0     420      .1       0
Bank Sta=157.56,244.12
XS Rating Curve= 0 ,0
Exp/Cntr=0.3,0.1

Type RM Length L Ch R = 1 ,61770   ,166,166,166
XS GIS Cut Line= 3
2381337.22003089692860.1279934972381652.10932462692681.888770628
 2381709.5419631692295.703787745
#Sta/Elev= 30
       0 2513.07      31 2500.27    63.1 2483.09    86.1 2473.71    99.9 2470.72
     110 2465.04   139.3 2465.32   152.2 2460.04   159.7    2459   186.3 2461.47
   215.7 2461.21   222.4 2458.65   236.2 2455.96   297.6 2456.07  316.01 2458.64
   325.1 2466.37   361.8 2490.07   423.2 2493.93   435.3 2492.61   451.5 2487.25
   468.1 2485.71   487.9 2487.46   516.2 2494.67   540.5 2508.04   552.6 2512.09
   605.2 2516.51   649.7 2515.64   726.5 2526.69   738.6    2531   752.3 2530.77
#Mann= 5 ,-1,0
       0      .1       0      20     .06       0     130      .1       0
   222.4    .045       0  316.01      .1       0
Bank Sta=222.4,316.01
XS Rating Curve= 0 ,0
Exp/Cntr(USF)=0,0
Exp/Cntr=0.3,0.1

Type RM Length L Ch R = 1 ,61604   ,351.6,351.6,351.6
XS GIS Cut Line= 4
2381390.77898477693006.0452314122381512.71979935692905.374898625
2381872.26926426  692835.74708512382047.60861571692863.675510899
#Sta/Elev= 30
       0 2530.45    22.6 2515.52    63.4 2494.26      83 2486.18   101.9 2471.27
   114.5 2464.58     147 2461.85   161.2 2463.53   181.7 2463.57   198.8    2459
   233.12457.516   251.3 2454.81   279.8 2454.47   308.3  2454.6  318.292457.514
   332.8 2468.34   338.7 2470.66     398 2471.14   426.5 2475.93   451.4 2477.78
   463.1 2481.76   483.5 2494.99   516.1 2496.66   532.2 2501.27   556.7 2503.57
   560.7 2504.58   572.9 2512.18   593.1 2519.87   625.5 2524.61   701.9 2544.51
#Mann= 6 ,-1,0
       0      .1       0      80     .06       0     130     .07       0
  198.13      .1       0   233.1    .045       0  318.29      .1       0
Bank Sta=233.1,318.29
XS Rating Curve= 0 ,0
Exp/Cntr=0.3,0.1

Type RM Length L Ch R = 1 ,61253   ,86.7,86.7,86.7
XS GIS Cut Line= 4
2381519.57194533693280.5249451082381601.45934227693241.989699489
2381843.91026262693206.6657243392382070.30483063693044.496565694
#Sta/Elev= 30
       0 2519.38     5.1 2513.38    18.3 2495.01    26.6 2486.78      30 2484.55
    49.3 2473.75    58.1 2470.03    71.4 2460.68    75.1 2459.29    97.1 2459.38
   113.5 2457.48   137.7 2456.67     143 2455.19   149.8 2452.94   174.1 2452.78
   218.6 2453.04  223.782455.188   230.7 2459.44   238.8 2466.82   250.9 2469.02
     263 2476.73   279.2 2479.39   340.8 2478.77   422.8 2481.71   468.6  2484.9
   496.1 2488.76   508.8 2488.96   537.6 2493.07   586.2 2511.49     614 2523.27
#Mann= 8 ,-1,0
       0      .1       0      30     .06       0   140.5     .07       0
     143    .045       0  223.78     .07       0   240.5      .1       0
  335.51     .05       0  455.51      .1       0
Bank Sta=143,223.78
XS Rating Curve= 0 ,0
Exp/Cntr(USF)=0,0
Exp/Cntr=0.3,0.1

Type RM Length L Ch R = 1 ,61166   ,53.4,53.4,53.4
XS GIS Cut Line= 4
2381527.04398067693326.1720558172381661.57290976693286.484594697
2381798.17929373693364.1794256012382132.10285396693101.743167076
#Sta/Elev= 30
       0 2531.84    14.6 2521.24      21 2515.14    27.5  2507.2    34.5 2493.47
    40.4 2486.61      50 2480.36    59.6  2476.5    80.4 2459.22   109.6 2457.94
   130.12454.446   166.3 2452.67   249.1 2452.77   264.4 2454.47   276.7 2459.84
   315.2 2461.41   330.5 2467.46   341.1 2468.47   366.1 2468.32   381.4 2474.54
   391.5 2476.38   429.2 2478.06   522.4 2478.84   544.2 2480.82   561.2 2480.14
   579.8 2481.29   588.7 2484.53   611.5 2488.17     640  2495.4   722.1 2525.36
#Mann= 7 ,-1,0
       0      .1       0      20     .06       0     130     .07       0
   130.1    .045       0   264.4      .1       0  357.42     .05       0
  477.42      .1       0
Bank Sta=130.1,264.4
XS Rating Curve= 0 ,0
Exp/Cntr=0.3,0.1

Type RM Length L Ch R = 1 ,61112   ,114,114,114
XS GIS Cut Line= 4
2381545.06703992693355.3655811482381648.33717084693325.150483113
 2381784.9435548693402.8453140172382143.49525905 693123.35880194
#Sta/Elev= 30
       0 2529.26    19.9 2512.43    28.2 2498.51    32.4 2493.36    40.7 2487.71
    55.9 2474.42    69.9 2459.98   107.6 2456.01   125.1 2453.05   131.9 2449.76
     140 2449.12   195.5 2449.01     229    2450  243.62 2453.02   259.3 2457.22
   282.5  2457.8   294.2 2460.75   314.5 2461.01   330.9 2464.05   360.1 2464.43
   380.4 2473.59   395.6 2475.74   532.6 2480.32   547.8 2482.78   566.8 2481.85
   593.4 2486.78   608.7 2487.41   624.5 2490.06   644.2 2495.73   719.4 2521.72
#Mann= 6 ,-1,0
       0     .06       0   107.6     .08       0   125.1    .045       0
  243.62      .1       0  334.75     .05       0  464.75      .1       0
Bank Sta=125.1,243.62
XS Rating Curve= 0 ,0
Exp/Cntr=0.3,0.1

Type RM Length L Ch R = 1 ,60998   ,606.3,606.3,606.3
XS GIS Cut Line= 3
2381599.85370704693519.7645949892381988.41743369693405.764493368
2382190.72747319693176.158654891
#Sta/Elev= 30
       0 2528.64    12.8 2520.51    21.2 2513.74    37.9 2497.49    46.2 2487.49
    58.7 2478.22    62.9 2473.42    71.2 2458.99    75.4 2457.03   104.5 2455.41
  112.722451.719   118.4 2448.99   129.6 2448.45   162.9 2448.63   183.8 2449.99
  189.772451.718   200.4 2456.39   242.1 2457.94   263.4 2460.14   342.2 2459.11
     363 2466.11   383.8 2475.15     388 2475.83     402 2476.18     476 2483.05
   490.2 2482.76   604.2 2489.94     651 2498.78   682.9 2507.96710.9616 2519.63
#Mann= 4 ,-1,0
       0      .1       0      50     .08       0  112.72    .045       0
  189.77      .1       0
Bank Sta=112.72,189.77
XS Rating Curve= 0 ,0
Exp/Cntr(USF)=0,0
Exp/Cntr=0.3,0.1

Type RM Length L Ch R = 1 ,60392   ,620,620,620
XS GIS Cut Line= 4
2381767.33932099694234.8396222752382112.54832099693938.434622275
2382347.47391969693731.3189490892382429.12459391693553.928923559
#Sta/Elev= 30
       0 2493.41    27.3 2482.55    41.5 2480.17    74.9 2469.83    88.5 2468.02
   222.5 2461.94     270 2462.27   293.9  2465.1   306.9 2462.75   321.8 2453.64
   347.8 2452.78   359.6  2447.1   367.7 2444.29   407.4 2443.89   422.9 2444.63
   430.1 2447.06   449.2 2450.51   529.2 2448.49   553.7 2450.78   583.9    2450
   622.8 2454.22   683.8 2456.35   694.5 2455.32   704.9 2458.04     723 2467.47
   736.2 2471.49   769.9  2473.6   871.8 2485.03   942.1 2499.05   963.5 2506.63
#Mann= 6 ,-1,0
       0      .1       0     100     .05       0     200      .1       0
     230     .06       0   359.6    .045       0   430.1      .1       0
Bank Sta=359.6,430.1
XS Rating Curve= 0 ,0
Exp/Cntr=0.3,0.1

Type RM Length L Ch R = 1 ,59772   ,581.9,581.9,581.9
XS GIS Cut Line= 3
2381983.48853553 694595.279043432382452.21778509694352.971848351
2382680.48786235694329.805392953
#Sta/Elev= 30
       0 2486.09    27.8 2482.23    50.3 2480.88    90.8 2476.22   109.1 2470.88
   126.7 2462.61   135.9 2461.81   149.4 2458.01   243.9 2456.39   346.4 2458.93
   356.5 2457.05   370.1 2447.58   374.5 2445.51     433 2443.69   482.9 2443.88
   527.5 2446.73   563.8 2443.59   582.8 2438.57     596 2436.03   624.1 2435.66
   648.2 2436.66  652.94 2438.55   656.3 2442.31   664.3  2454.7   672.4 2462.46
   680.4  2472.3   688.4 2479.62   700.5 2487.85   720.6 2499.05   757.1 2523.48
#Mann= 7 ,-1,0
       0      .1       0     180     .05       0     400     .06       0
     420     .07       0     510      .1       0   582.8    .045       0
  652.94      .1       0
#XS Ineff= 2 , 0
           534.5    2450
Permanent Ineff=
       F       F
Bank Sta=582.8,652.94
XS Rating Curve= 0 ,0
Exp/Cntr=0.3,0.1

Type RM Length L Ch R = 1 ,59190   ,438.5,438.5,438.5
XS GIS Cut Line= 3
2381976.84146939694858.5821549712382135.00971603694914.703253209
2382749.09907853694922.368967154
#Sta/Elev= 30
       0 2494.07    54.5 2470.67    79.9 2462.63    92.7 2460.23   143.6 2455.24
     181 2449.88     205 2448.86     237 2450.75   357.1 2451.69     453  2446.4
     501 2446.24     517 2446.97     533 2442.77     557 2443.56     577  2438.6
  592.472432.629     613 2430.19   636.4 2429.95   656.7 2430.49     665 2432.63
     669 2434.26     681 2450.24   693.1 2461.08   716.7  2486.6     721 2492.03
     733 2501.33     741 2506.24     749 2512.96     769 2526.08     782 2537.99
#Mann= 6 ,-1,0
       0      .1       0  167.83     .05       0  467.83     .06       0
  592.47    .045       0     665     .06       0  667.83      .1       0
Bank Sta=592.47,665
XS Rating Curve= 0 ,0
Exp/Cntr=0.3,0.1

Type RM Length L Ch R = 1 ,58752   ,521.7,521.7,521.7
XS GIS Cut Line= 3
 2381923.2145109695184.3535544932382649.02129919695391.598700806
2382738.30053926695396.213240071
#Sta/Elev= 30
       0 2483.89    71.7  2459.9    92.5 2456.55   138.3 2452.29     209 2449.46
   300.5 2450.58   329.6 2449.75   342.1    2447   362.9 2437.75     380 2437.56
   433.6  2437.2   462.7 2439.91   504.3 2438.83   512.7 2440.25   528.9 2440.26
   554.3 2438.84   558.4 2437.79  566.042429.447   571.2 2426.96   633.3 2426.73
   641.6 2426.81  652.382429.443   674.5 2433.76   690.7 2434.32   724.8 2437.44
   741.5 2440.69   749.8 2445.09     786 2469.42   801.2 2476.69   844.2 2502.07
#Mann= 7 ,-1,0
       0      .1       0     120     .05       0     330      .1       0
     380     .05       0     430     .06       0  566.04    .045       0
  652.38      .1       0
Bank Sta=566.04,652.38
XS Rating Curve= 0 ,0
Exp/Cntr=0.3,0.1

Type RM Length L Ch R = 1 ,58230   ,504.1,504.1,504.1
XS GIS Cut Line= 3
 2381924.0252335 695729.664995522382536.89042193695900.798654977
 2382611.9750851695901.801532696
#Sta/Elev= 30
       0 2464.94    25.7 2458.74    41.7 2456.63    72.6 2450.91   120.6 2445.68
   128.9 2442.63   137.2 2438.14   149.7  2433.1     158 2431.23     187 2431.36
   216.1 2433.96   257.6 2434.16   307.5 2432.99   340.7 2434.91   378.1 2435.06
   407.2 2433.56   411.3 2431.78   419.6 2425.93   423.8  2423.7   427.9 2423.36
   486.1  2423.3   506.8 2424.22  516.62 2425.96   523.4 2428.59   527.6 2429.23
   606.5    2429   639.6 2433.31   643.9 2435.48   683.6 2464.46   711.4 2480.96
#Mann= 5 ,-1,0
       0      .1       0     220     .05       0     330     .06       0
   419.6    .045       0  516.62      .1       0
#XS Ineff= 2 , 0
           343.1 2439.16
Permanent Ineff=
       F       F
Bank Sta=419.6,516.62
XS Rating Curve= 0 ,0
Exp/Cntr=0.3,0.1

Type RM Length L Ch R = 1 ,57726   ,497.6,497.6,497.6
XS GIS Cut Line= 2
 2382067.5475109696466.741960584 2382618.2211484 696254.83616811
#Sta/Elev= 30
       0 2451.95    17.8 2449.47    30.7 2446.31    43.5 2441.77    69.2 2428.21
    77.8 2426.25    97.6 2424.97   116.2 2425.99   202.1 2425.66   227.8 2426.25
   249.3  2428.4   262.1 2428.22   287.8 2426.58  297.722421.149     305 2418.03
   326.4 2417.91   347.8 2418.17  362.852421.147   382.1 2425.12   463.6 2425.64
   480.7 2423.95   490.7 2421.97   502.1 2422.45   510.7  2424.7   519.3 2429.26
   532.1 2438.83     545 2444.18   570.7 2459.38   583.6 2464.25     590 2468.03
#Mann= 6 ,-1,0
       0     .05       0     180     .06       0     290     .05       0
  297.72    .045       0  362.85     .05       0     390      .1       0
#XS Ineff= 2 , 0
           249.3    2430
Permanent Ineff=
       F       F
Bank Sta=297.72,362.85
XS Rating Curve= 0 ,0
Exp/Cntr=0.3,0.1

Type RM Length L Ch R = 1 ,57228   ,625.6,625.6,625.6
XS GIS Cut Line= 4
2382298.98213317696995.5242597792382414.39968767696948.671203046
2382699.87671455696715.7301181022382771.94964616696687.079399522
#Sta/Elev= 30
       0 2465.53    44.5 2462.37    61.1 2459.39    67.2  2456.1     104 2431.14
   116.3 2425.41   122.2 2423.98     132 2423.87   147.5 2422.13   212.3 2421.56
   227.8 2420.43   250.8 2422.47   269.3 2421.07   281.7 2417.75   292.1 2419.85
   302.4 2418.74   313.1  2419.1   364.2 2417.23   379.8 2415.08   455.2 2414.67
   462.4 2414.96   471.7 2417.22   486.5  2422.1   507.5 2438.64   519.2 2445.77
   523.5  2447.2   527.8 2449.76   543.2 2463.04   550.7 2468.23   570.6 2484.51
#Mann= 5 ,-1,0
       0     .05       0  154.56      .1       0  264.56     .06       0
   364.2    .045       0   471.7      .1       0
#XS Ineff= 2 , 0
           245.6    2430
Permanent Ineff=
       F       F
Bank Sta=364.2,471.7
XS Rating Curve= 0 ,0
Exp/Cntr=0.3,0.1

Type RM Length L Ch R = 1 ,56603   ,551.1,551.1,551.1
XS GIS Cut Line= 3
2382358.42228661697390.8829757082382477.42245029697457.978504787
2382992.12106241697303.567997151
#Sta/Elev= 30
       0 2443.47    45.4 2439.81    94.3 2433.94    99.9 2432.37   126.3    2422
   135.4 2420.54   165.2 2419.28     223 2419.28   256.4 2417.98   327.4 2421.56
   344.1 2420.55   360.8 2417.25   369.2 2416.66   452.7 2419.16   481.9 2417.38
   486.1 2416.68   492.8 2414.25  510.242411.361   519.5 2409.54     532 2408.86
   594.7 2408.93   602.1 2409.86  605.722411.359   611.7 2415.06   615.6 2418.63
   628.7 2432.76   636.4 2439.46     647 2447.31   657.3 2453.36     674 2461.01
#Mann= 7 ,-1,0
       0     .05       0      90      .1       0  196.61     .05       0
  396.61     .06       0  506.61      .1       0  510.24    .045       0
  605.72      .1       0
#XS Ineff= 2 , 0
        437.2264    2430
Permanent Ineff=
       F       F
Bank Sta=510.24,605.72
XS Rating Curve= 0 ,0
Exp/Cntr=0.3,0.1

Type RM Length L Ch R = 1 ,56052   ,497,497,497
XS GIS Cut Line= 3
2382614.91366741697904.9246973582383091.21156069697870.558062124
2383172.52318637697804.078722208
#Sta/Elev= 30
       0 2442.91    25.3 2440.31    37.4 2438.04    61.4  2426.2    73.5 2421.37
    81.5 2416.92    85.5 2416.18   146.8 2414.13   245.9 2413.83     274 2414.75
     298  2413.7   306.1 2414.32   310.1 2413.72   318.1 2408.52  322.072406.912
   330.1 2404.94   374.2 2404.62   398.3 2404.95  406.372406.911   418.3  2409.7
   464.8 2412.36   478.8 2414.19   483.9 2416.04   492.4 2421.44   499.4 2424.52
   521.8 2433.55   536.1 2437.12   561.9 2447.04   571.8 2451.12   582.6 2457.24
#Mann= 5 ,-1,0
       0     .05       0     310     .06       0  322.07    .045       0
  406.37     .06       0     410      .1       0
Bank Sta=322.07,406.37
XS Rating Curve= 0 ,0
Exp/Cntr=0.3,0.1

Type RM Length L Ch R = 1 ,55555   ,495,495,495
XS GIS Cut Line= 3
2382544.60228289698446.8536030612382994.06928289698376.151603061
2383444.35128289698310.554603061
#Sta/Elev= 30
       0 2456.96    25.6 2448.09      32  2443.8    44.1 2433.09    48.2 2431.86
    68.4 2432.01    80.6 2430.25   108.9 2411.06     117 2408.07   129.1 2406.09
     204 2405.55   246.6 2407.94   424.7  2409.1   428.8 2408.34   434.9 2403.05
   440.9 2399.85   457.1 2399.61   485.4 2400.22  495.852403.052   517.8 2408.95
   554.1 2405.52   594.6 2405.96   610.7 2404.87   655.2 2410.17   683.5 2410.25
     732 2407.58   792.6 2407.32   804.8 2411.59   829.9  2423.7     910 2450.38
#Mann= 8 ,-1,0
       0      .1       0      60     .06       0      90     .05       0
     390     .06       0   434.9    .045       0  495.85      .1       0
  684.99     .06       0  784.99      .1       0
#XS Ineff= 2 , 0
        381.8464    2412
Permanent Ineff=
       F       F
Bank Sta=434.9,495.85
XS Rating Curve= 0 ,0
Exp/Cntr=0.3,0.1

Type RM Length L Ch R = 1 ,55060   ,319.6,319.6,319.6
XS GIS Cut Line= 3
 2382761.5911647698997.1961819162383361.92867569698756.708231615
2383448.46391176 698776.33218924
#Sta/Elev= 30
       0 2446.27    11.4 2439.04    48.1 2410.08    54.5 2406.66    63.5 2407.17
    94.3 2404.96   109.7 2401.88   213.1 2403.68   282.9  2403.4     326  2404.8
   334.6  2405.9   377.7 2403.29     382 2401.97  386.282399.242   394.9 2396.67
   408.8 2396.49   450.9 2396.71  458.41 2399.24   463.8    2401   485.4 2399.26
   503.5 2399.72   537.9 2401.65     563  2404.2   617.3 2405.62   627.6 2406.94
   636.2 2409.46   644.8 2413.74   657.2 2422.36   673.6 2431.48   735.4 2457.14
#Mann= 8 ,-1,0
       0     .06       0      70     .05       0     180     .07       0
     280      .1       0  386.28    .045       0  458.41      .1       0
     500     .06       0     600      .1       0
Bank Sta=386.28,458.41
XS Rating Curve= 0 ,0
Exp/Cntr=0.3,0.1

Type RM Length L Ch R = 1 ,54740   ,152.5,152.5,152.5
XS GIS Cut Line= 3
2382838.61221327699185.0371427212383333.33829462699138.463804332
2383399.82289193699082.458400351
#Sta/Elev= 30
       0 2440.42    13.6 2433.81    21.7 2426.27    25.7 2423.99    41.7 2422.96
    57.8  2411.5    73.9 2402.08    81.9 2399.71      90 2400.66     102 2403.38
   114.1 2404.11   122.5 2406.64   146.2 2406.85   182.4 2405.12   210.5 2399.72
   250.3  2400.2   294.9 2403.56     331 2403.26     335 2402.08  342.74 2396.13
   351.1 2393.96   383.2 2393.94   427.3 2394.38  432.98 2396.13   447.5 2402.58
   463.6 2413.42   471.3 2415.81   496.9 2417.38   536.2 2426.45   583.8 2430.99
#Mann= 7 ,-1,0
       0      .1       0      90     .06       0     190     .07       0
     290     .05       0  342.74    .045       0  432.98     .08       0
     480     .06       0
#XS Ineff= 2 , 0
           130.4 2411.92
Permanent Ineff=
       F       F
Bank Sta=342.74,432.98
XS Rating Curve= 0 ,0
Exp/Cntr(USF)=0,0
Exp/Cntr=0.3,0.1

Type RM Length L Ch R = 1 ,54588   ,97.2,97.2,97.2
XS GIS Cut Line= 4
2382836.98646901699213.2954726962383104.24437669699220.778886173
2383325.90282938 699365.77283374 2383489.9594887 699359.27277506
#Sta/Elev= 30
       0 2440.81    19.2 2428.85    31.2  2427.3    41.9 2419.89    59.2 2410.32
    95.2 2398.38   135.2 2399.27   167.3 2407.33   207.3 2407.04   231.3  2405.5
   266.9 2399.11   329.4 2398.02  349.87 2394.11   363.1 2392.12   406.9 2391.87
     425 2392.09   429.8 2394.15   434.6 2397.84   444.1 2407.56   448.9 2410.45
   487.1 2411.29   496.7 2413.73   516.1 2413.52   525.4    2417   546.5 2429.67
   562.5 2435.16   570.5 2436.69   630.6 2440.33   662.6 2439.11   696.4 2443.64
#Mann= 7 ,-1,0
       0      .1       0      90     .06       0     190     .07       0
  349.87    .045       0   429.8     .08       0  527.36     .07       0
  622.23      .1       0
#XS Ineff= 2 , 0
          170.32 2410.86
Permanent Ineff=
       F       F
Bank Sta=349.87,429.8
XS Rating Curve= 0 ,0
Exp/Cntr=0.3,0.1

Type RM Length L Ch R = 1 ,54490   ,156.6,156.6,156.6
XS GIS Cut Line= 4
2382830.39963007699286.7584097552383013.68070948699287.583484462
 2383316.8014847699462.8889938982383442.96869168699420.393955499
#Sta/Elev= 30
       0 2445.92     5.8 2440.68    17.8 2438.87    21.8 2436.93    29.8 2431.51
    49.8 2419.99    77.8 2406.95    85.8 2400.99    93.8 2397.91   117.8 2397.09
   223.1 2398.79   285.8  2400.9   315.5 2399.18   332.7 2392.71   343.3 2391.03
   379.5 2390.07     408 2390.65  413.51 2392.79   435.1 2404.39     441 2406.65
     505 2405.47   556.4 2406.56   597.4 2405.83   608.8 2408.46     614 2411.14
   621.4 2416.12   625.6 2417.79   629.9 2418.62   638.5 2421.97   666.6 2429.11
#Mann= 12 ,-1,0
       0      .1       0     100     .06       0  193.28     .07       0
  263.28      .1       0  313.28     .07       0   332.7    .045       0
  413.51     .07       0  423.28     .08       0  453.28     .07       0
  533.28     .08       0  643.45     .07       0  663.45      .1       0
#XS Ineff= 2 , 0
          284.04  2403.4
Permanent Ineff=
       F       F
Bank Sta=332.7,413.51
XS Rating Curve= 0 ,0
Exp/Cntr=0.3,0.1

Type RM Length L Ch R = 1 ,54334   ,359.7,359.7,359.7
XS GIS Cut Line= 4
2382806.87593593699454.9225276652382910.39425692699446.112457794
2383336.47356805699615.3982579712383436.27224907699438.180318965
#Sta/Elev= 30
       0 2476.56    25.4 2458.44    41.4 2444.32    57.5 2442.12    73.6 2427.86
      99 2408.96     123 2397.06   135.9 2395.21   200.5 2397.18   234.9 2394.29
   264.7 2395.84   290.9 2395.25   303.8 2394.24   312.4    2392   329.4 2389.01
     354 2388.86   381.3 2389.01  389.34 2392.03   394.4 2396.13   403.3 2400.89
   536.2 2397.47   575.5 2399.04   587.9 2403.11   592.5 2403.41   670.5 2403.56
   707.2 2405.38   734.8 2404.56     744 2406.86   760.5 2420.79   765.8 2423.21
#Mann= 5 ,-1,0
       0      .1       0   312.4    .045       0  389.34      .1       0
  543.89     .08       0  722.37     .07       0
#XS Ineff= 2 , 0
          201.01 2411.21  409.53         2411.66
Permanent Ineff=
       F       F
Bank Sta=312.4,389.34
XS Rating Curve= 0 ,0
Exp/Cntr(USF)=0,0
Exp/Cntr=0.3,0.1

Type RM Length L Ch R = 1 ,53974   ,332.1,332.1,332.1
XS GIS Cut Line= 3
2383055.08797192699942.9782629712383535.28403627699498.114915731
2383560.68674893699445.738917953
#Sta/Elev= 30
       0 2443.29    12.4 2441.68    32.1 2437.02    43.8 2426.37    61.5 2407.06
    64.3 2403.24    72.4 2389.14   73.66 2388.04    77.8 2386.01    84.1 2385.19
   114.5 2384.84   135.1 2385.36  144.66 2388.04   152.1 2392.52   155.7 2393.59
     176 2392.57   208.7 2392.38   273.8 2395.73   317.7 2396.85   409.6 2395.51
   446.4  2398.4   532.4 2397.79   538.3 2398.26     550 2402.27   561.8 2402.88
   644.2 2402.49     656 2406.29     669 2416.63   677.9 2424.99   712.8  2442.1
#Mann= 7 ,-1,0
       0      .1       0   73.66    .045       0  144.66      .1       0
     230     .06       0     480     .08       0     490     .05       0
     630     .07       0
Bank Sta=73.66,144.66
XS Rating Curve= 0 ,0
Exp/Cntr=0.3,0.1

Type RM Length L Ch R = 1 ,53642   ,637,637,637
XS GIS Cut Line= 2
2383386.20570808700150.0529140312383633.38662638699465.400237425
#Sta/Elev= 30
       0 2441.28    43.5 2435.83      52 2433.22    61.6 2426.88    73.2 2416.55
   108.5 2389.04   115.8 2384.54  123.572382.114     137 2379.16   145.5 2380.02
   162.5 2379.18   196.6 2379.38   200.8 2380.03  203.912382.116   209.3 2386.28
   217.8 2388.34   295.9  2390.1   366.7 2389.57   406.3 2391.55   559.4 2396.27
   570.8 2397.25   583.4  2400.3   604.8 2399.85   660.1 2401.38   664.4 2402.98
   667.8 2405.79   681.4 2419.85   685.6 2423.19   711.1 2437.47   727.9 2445.28
#Mann= 7 ,-1,0
       0      .1       0  123.57    .045       0  203.91     .06       0
     380     .05       0     460     .07       0     570     .08       0
     670     .06       0
Bank Sta=123.57,203.91
XS Rating Curve= 0 ,0
Exp/Cntr=0.3,0.1

Type RM Length L Ch R = 1 ,53005   ,454,454,454
XS GIS Cut Line= 2
2383914.99803915700543.3456902092384238.13311745699693.086729358
#Sta/Elev= 30
       0 2414.47    49.4 2406.48   130.7 2397.44   207.2 2392.91   276.2    2391
   284.8 2388.87     291 2384.61   298.5 2377.58   301.9 2375.37   306.1 2374.86
   357.5  2374.7   383.2 2374.95   388.2 2377.58   393.3 2382.15   400.3 2384.91
     570 2381.82   652.7 2380.99   682.7  2381.8   695.5 2380.56   806.8 2381.44
   811.9 2382.46   823.9 2388.87   828.2 2389.86   864.6 2390.52   866.7 2391.35
   870.8 2394.93   879.5 2404.35   883.2 2407.07   896.7 2412.06   909.6 2421.78
#Mann= 11 ,-1,0
       0      .1       0     150     .05       0     260      .1       0
   298.5    .045       0   388.2      .1       0     470     .05       0
     570     .07       0     680     .05       0     780     .06       0
     810     .08       0     890     .06       0
#XS Ineff= 1 ,-1
   402.6 909.591    2386
Permanent Ineff=
       F
Bank Sta=298.5,388.2
XS Rating Curve= 0 ,0
Exp/Cntr=0.3,0.1

Type RM Length L Ch R = 1 ,52551   ,520,520,520
XS GIS Cut Line= 2
2384322.09920314700836.6521299552384635.99131931699822.622364083
#Sta/Elev= 30
       0  2393.3    10.8 2390.15    42.8 2386.11    90.8 2385.14   104.1 2382.41
   116.3 2384.19   426.5 2384.69   434.9 2383.97   450.62376.002     460 2370.96
   496.8 2370.58     527 2370.78   532.82372.974   543.8 2376.61   623.3 2380.95
   765.4  2378.4   774.1 2380.35   782.5 2377.81   845.3  2379.2   920.6 2377.34
   926.9 2378.83   938.1 2386.69   945.8 2389.59   979.7 2389.39  1000.2  2405.1
  1012.8 2408.12  1024.4 2420.65  1030.8 2424.77  1037.9 2427.64  1061.5  2430.8
#Mann= 7 ,-1,0
       0      .1       0     150     .05       0     350     .06       0
   450.6    .045       0   532.8      .1       0     660     .06       0
     970      .1       0
#XS Ineff= 2 , 0
                          620.36         2385.64
Permanent Ineff=
       F       F
Bank Sta=450.6,532.8
XS Rating Curve= 0 ,0
Exp/Cntr=0.3,0.1

Type RM Length L Ch R = 1 ,52031   ,99.1,99.1,99.1
XS GIS Cut Line= 3
2384934.46164088  701244.58260332384999.87640967700130.549268033
2385017.71680116700094.868485053
#Sta/Elev= 30
       0 2412.15    11.4 2402.95    39.5  2384.3    67.5 2376.82   119.6 2380.14
   163.7 2381.47   235.9 2377.94   259.9 2377.83   271.9  2379.2     356 2378.29
     364 2376.76   465.8 2379.39   659.6    2378   684.6 2376.93   735.3 2378.53
   760.7 2377.92   773.5 2370.67   780.7 2367.55   784.8 2367.25   828.8 2367.08
   841.3 2367.91  854.53 2370.67   892.9 2373.19   977.1    2375  1049.2 2374.09
  1101.3 2374.86  1109.3 2376.49  1113.3 2378.49  1132.1 2391.251155.845  2391.9
#Mann= 8 ,-1,0
       0      .1       0      60     .06       0     250     .05       0
   773.5    .045       0  854.53      .1       0     940     .05       0
    1040     .06       0 1145.95     .07       0
Bank Sta=773.5,854.53
XS Rating Curve= 0 ,0
Exp/Cntr(USF)=0,0
Exp/Cntr=0.3,0.1

Type RM Length L Ch R = 1 ,51932   ,44.2,44.2,44.2
XS GIS Cut Line= 4
2385018.58785732701247.1357809982385073.63774245700482.762831397
2385109.94008811700242.4460267542385129.54384847  700143.9852495
#Sta/Elev= 30
       0  2402.9    42.1 2379.03    54.1 2376.26   151.7 2378.74   190.4 2378.16
   233.8 2375.71   294.7 2377.39     415 2376.05   463.2 2377.92   534.5 2375.44
   575.4 2376.32   623.6 2375.09   684.2  2377.1   740.3 2376.36   751.9 2378.15
     768 2376.39  778.35 2369.08   784.1 2366.18   808.1 2365.86   840.8 2366.06
  851.57 2369.08   873.1 2370.36   885.3 2373.85   925.7 2372.62    1043 2372.88
  1059.6 2374.35  1067.8 2378.91  1080.4 2381.98  1092.3 2389.09  1109.8 2389.22
#Mann= 6 ,-1,0
       0      .1       0     160     .06       0     450     .05       0
     650     .06       0  778.35    .045       0  851.57     .06       0
Bank Sta=778.35,851.57
XS Rating Curve= 0 ,0
Exp/Cntr=0.3,0.1

Type RM Length L Ch R = 1 ,51888   ,97.9,97.9,97.9
XS GIS Cut Line= 4
2385060.86925187701253.358703616  2385115.919137700488.985754015
2385152.22148266700248.6689493712385171.82524302700150.208172118
#Sta/Elev= 30
       0 2397.39    20.2 2382.38    28.3 2378.85    36.9 2377.74   116.5 2378.84
   192.7 2377.89   228.8 2374.32   252.8 2373.71   272.6 2376.55   345.1 2377.58
   481.4 2374.32   513.5 2376.04   525.5 2375.18   565.6 2376.02   598.1 2375.35
   699.1 2376.95   782.3 2374.39   786.4 2373.21  793.04  2368.6   798.5 2365.95
   802.6 2365.62     843 2365.69   863.2 2368.61   923.9 2371.94   999.3 2371.91
  1057.8 2374.38    1066 2375.91  1078.2  2385.7  1082.3 2387.62  1109.8  2387.7
#Mann= 4 ,-1,0
       0      .1       0     160     .06       0  793.04    .045       0
   863.2     .06       0
#XS Ineff= 2 , 0
          512.92 2379.13
Permanent Ineff=
       F       F
Bank Sta=793.04,863.2
XS Rating Curve= 0 ,0
Exp/Cntr=0.3,0.1

Type RM Length L Ch R = 1 ,51790   ,660.7,660.7,660.7
XS GIS Cut Line= 4
2385126.98785344701227.5599329392385241.70881231700624.810070211
2385213.96034712700343.2543845892385274.27624548700147.689329559
#Sta/Elev= 30
       0 2384.88    18.7 2385.04    83.9 2377.73   153.1 2373.87   324.1 2376.84
   523.6 2373.24   609.1 2374.54   710.8 2371.52   757.9 2371.64   765.9 2372.06
     774 2373.77     782 2372.74   799.4 2368.43   806.1  2365.7   830.2 2365.62
   850.3 2365.81   869.22368.409   899.9  2370.7     928 2371.66  1007.5 2371.62
  1011.7 2373.02  1018.3 2377.02  1028.4 2378.85  1036.8 2384.09  1039.7 2384.73
  1074.5 2384.47  1078.7 2386.98    1087 2393.56  1095.1 2397.23  1101.1 2401.73
#Mann= 7 ,-1,0
       0      .1       0      40     .05       0  643.57     .06       0
   799.4    .045       0   869.2      .1       0  936.49     .06       0
 1036.49     .07       0
#XS Ineff= 2 , 0
          609.87 2380.64
Permanent Ineff=
       F       F
Bank Sta=799.4,869.2
XS Rating Curve= 0 ,0
Exp/Cntr(USF)=0,0
Exp/Cntr=0.3,0.1

Type RM Length L Ch R = 1 ,51129   ,227.7,227.7,227.7
XS GIS Cut Line= 2
2385601.12719103701019.2294564012385939.57159516700273.842742424
#Sta/Elev= 30
       0 2387.58    28.6 2386.75    50.6 2379.75    76.9 2369.96    98.9 2367.52
   107.7 2367.83   120.9 2366.68     134 2367.33   419.6 2365.68   498.7 2368.05
   529.4  2368.1   539.5 2369.71   542.6 2369.21  553.75 2361.14   560.2 2358.89
   586.9 2359.36   605.1 2357.57   612.9 2357.82   621.7 2361.08   630.5 2361.88
   639.2 2365.52   652.4 2368.38   661.2 2376.02     670 2381.09   680.6 2382.09
   707.8 2381.89   716.9  2382.7   740.3 2388.11   775.4  2401.5   818.6 2410.93
#Mann= 5 ,-1,0
       0     .05       0     460     .06       0  553.75    .045       0
   621.7     .06       0     680      .1       0
#XS Ineff= 2 , 0
         145.479    2380
Permanent Ineff=
       F       F
Bank Sta=553.75,621.7
XS Rating Curve= 0 ,0
Exp/Cntr=0.3,0.1

Type RM Length L Ch R = 1 ,50902   ,99.4,99.4,99.4
XS GIS Cut Line= 3
2385754.96664398 701035.688368272385800.79851196701014.356803898
2386109.03935773700474.264638845
#Sta/Elev= 30
       0 2388.35    24.9 2386.23    32.2 2383.97    41.9 2378.77    53.9 2374.34
    73.5 2372.62    89.6 2369.18   105.8 2369.79   121.9 2372.91   146.1  2369.6
   208.5 2367.29   262.1 2366.89   286.8 2364.11     319 2362.38   378.9 2361.88
   440.9 2365.19   511.3 2364.81   520.1 2363.76  529.252359.521   535.5 2356.82
   540.1 2356.21   576.9  2355.9     590 2357.69  593.262359.518     600 2363.45
   613.8 2367.91   625.7 2376.79   641.4 2378.74   655.2 2387.82   672.4  2388.5
#Mann= 6 ,-1,0
       0     .05       0      30     .06       0   80.55     .05       0
  400.55     .06       0  529.25    .045       0  593.26     .06       0
Bank Sta=529.25,593.26
XS Rating Curve= 0 ,0
Exp/Cntr=0.3,0.1

Type RM Length L Ch R = 1 ,50802   ,25.9,25.9,25.9
XS GIS Cut Line= 3
2385883.33477964701176.4595440872385860.86155159701040.948777821
 2386232.9041322700481.456346046
#Sta/Elev= 30
       0 2394.25    43.9 2381.94   116.9 2373.78   137.4 2374.44   223.6 2369.41
   309.8 2366.75   348.4 2363.92   390.6 2362.74   483.1 2362.82   511.8 2364.75
   562.3 2364.95   593.4  2368.4   608.6 2358.85   617.4 2355.49   631.9 2355.23
   661.8 2356.01  671.37 2358.83   679.1 2368.66     682 2370.99   685.1 2372.16
   705.1 2372.59   716.6 2374.93   718.3 2375.65   728.2 2385.13   733.9 2388.22
   751.2 2391.06   785.9 2391.23   790.4 2393.09   800.7 2401.09   809.3 2404.02
#Mann= 7 ,-1,0
       0     .06       0      60     .05       0      90     .06       0
  317.36     .05       0  347.36     .06       0   608.6    .045       0
  671.37     .06       0
Bank Sta=608.6,671.37
XS Rating Curve= 0 ,0
Exp/Cntr=0.3,0.1

Type RM Length L Ch R = 1 ,50776   ,147.9,147.9,147.9
XS GIS Cut Line= 3
2385909.15709704701181.550684997 2385877.2115059701063.090172283
2386249.25408651700503.597740508
#Sta/Elev= 30
       0 2394.91    23.9 2392.29    58.4 2382.04    79.1    2378     125 2373.79
   168.2 2372.64   225.9 2368.43   388.1    2362   470.8 2361.64     507 2364.57
   547.7 2364.82   583.1 2367.21   590.4 2364.46   597.6 2358.54  611.04 2357.77
   619.3 2355.26   658.2 2354.57     663 2355.01   665.7 2357.76   672.6 2365.87
   677.4 2368.68   696.6 2370.15   706.1 2377.98   715.8 2380.08   725.4 2387.21
   730.2 2389.41   746.5  2391.7   785.4 2392.01   787.9 2392.49   794.6 2397.15
#Mann= 4 ,-1,0
       0     .06       0  611.04    .045       0   665.7      .1       0
  682.69     .06       0
Bank Sta=611.04,665.7
XS Rating Curve= 0 ,0
Exp/Cntr=0.3,0.1

Type RM Length L Ch R = 1 ,50628   ,362.9,362.9,362.9
XS GIS Cut Line= 4
2386036.62468656701152.0539662432386030.29378254701098.241282108
2386335.75990131700640.8334669612386343.67353133700569.610796782
#Sta/Elev= 30
       0 2388.83      15 2387.74      23    2386    39.1 2378.32    51.2 2370.42
    55.5 2369.26    65.1 2368.74    98.8 2362.13   122.4 2360.16   272.6 2359.89
   307.2    2359   316.9 2359.31   339.2 2362.06   440.3 2361.33   457.2 2362.71
   460.1  2362.5   471.6 2356.78   475.3  2354.8   483.5 2353.92   532.2 2354.35
  551.45  2356.8   572.5 2365.01   584.1 2366.93   589.4 2368.63   598.5 2373.14
   604.3 2374.24   611.9 2378.73     624 2382.34   640.1 2393.08   675.9 2395.08
#Mann= 7 ,-1,0
       0     .05       0   64.18     .06       0  134.18     .05       0
  414.18      .1       0   471.6    .045       0  551.45      .1       0
  644.21     .06       0
Bank Sta=471.6,551.45
XS Rating Curve= 0 ,0
Exp/Cntr(USF)=0,0
Exp/Cntr=0.3,0.1

Type RM Length L Ch R = 1 ,50266   ,465.2,465.2,465.2
XS GIS Cut Line= 3
2386139.05135476701367.2564401412386233.00787667701345.026275214
2386788.21890613700682.329785776
#Sta/Elev= 30
       0 2390.28     5.3 2389.49    13.5 2385.95    42.3 2366.95    58.7 2364.32
   127.7 2361.76   207.4  2363.2   237.2 2359.32   252.9 2358.57   319.5 2360.84
   385.5 2355.21   490.5 2359.35   534.7 2359.93   550.3 2359.14  569.282354.914
   581.4  2351.9   607.7 2351.41   643.4 2351.56  657.112354.914   670.4 2358.44
   768.8 2358.27   800.8  2360.1   811.3 2362.16   837.4 2379.09   868.7 2401.39
   879.1 2404.92   910.4 2406.77   919.3 2415.02   931.3 2424.01   961.1 2440.31
#Mann= 6 ,-1,0
       0     .05       0  556.55      .1       0  569.28    .045       0
  657.11      .1       0  816.55     .06       0  936.55      .1       0
#XS Ineff= 2 , 0
          203.61 2371.07
Permanent Ineff=
       F       F
Bank Sta=569.28,657.11
XS Rating Curve= 0 ,0
Exp/Cntr=0.3,0.1

Type RM Length L Ch R = 1 ,49801   ,736.7,736.7,736.7
XS GIS Cut Line= 2
2386332.07148224701817.4517364722387141.08363687 701022.43622746
#Sta/Elev= 30
       0 2371.32      54 2368.61    73.1    2365   103.1 2363.07     223 2357.76
   342.2  2355.9   415.1 2359.12   471.2 2359.75   531.1 2357.63     566  2358.8
   605.8 2357.09   701.2 2360.51   734.8 2359.55     747 2360.36   765.1 2351.52
   774.1 2349.04  797.08 2351.71     829 2348.56     863 2348.99   869.4 2351.74
   874.3 2354.65   879.9 2355.37   993.4 2353.25  1010.1 2353.81  1029.9 2356.52
  1041.2 2360.87  1054.5 2369.14  1072.3 2377.56  1103.4 2398.75  1134.3 2401.97
#Mann= 6 ,-1,0
       0      .1       0     190     .05       0     610      .1       0
  797.08    .045       0   869.4      .1       0    1040     .06       0
#XS Ineff= 2 , 0
          746.86 2365.68
Permanent Ineff=
       F       F
Bank Sta=797.08,869.4
XS Rating Curve= 0 ,0
Exp/Cntr=0.3,0.1

Type RM Length L Ch R = 1 ,49064   ,447.9,447.9,447.9
XS GIS Cut Line= 5
2386416.12100874701986.6464125122386619.13839269 701808.10538873
2387304.90317279 701818.839915792387457.39697998701817.875302334
2387529.31721172701783.489261371
#Sta/Elev= 30
       0 2402.19    32.3 2389.27      64  2365.4    90.6 2359.89   250.6 2356.62
   384.1  2351.3   487.4 2353.68   543.4 2351.85   623.4  2354.7   699.4 2352.73
   739.5 2354.53   775.5 2351.35   831.5 2353.08   839.6 2349.66   847.4 2348.32
   875.5 2346.36   887.5 2348.34   915.5 2347.27   923.5 2348.28  935.222344.437
   951.5 2341.11   995.5  2341.3 1004.122344.437  1019.5 2350.18  1035.5 2353.03
  1079.5 2357.91  1107.5 2357.17  1119.6 2358.94  1165.3  2386.3  1188.4 2388.08
#Mann= 7 ,-1,0
       0      .1       0     160     .05       0  810.36      .1       0
  935.22    .045       0 1004.12      .1       0 1106.21     .07       0
 1188.42     .06       0
Bank Sta=935.22,1004.12
XS Rating Curve= 0 ,0
Exp/Cntr=0.3,0.1
