HEC-RAS study DRKFK_2.prj: DRKFK_2

--- DRKFK_2.g01 (geometry) --- (continued)

Type RM Length L Ch R = 1 ,31394   ,441.1,441.1,441.1
XS GIS Cut Line= 3
2394210.86210575 714795.822206242394238.10503039714680.458756078
2394151.20086796714067.506758132
#Sta/Elev= 30
       0 2273.11    27.4 2261.16    60.3  2248.6      89 2234.62    93.1 2230.85
     103 2217.39   109.6 2212.74     138 2214.43   158.2 2211.19   251.1 2212.21
   261.1 2211.46   287.5 2208.97   348.1 2209.91  355.49 2211.45   368.3 2217.29
   416.7 2219.91   420.8 2218.94   432.9 2211.65     441 2209.93   487.6 2211.78
   550.1 2211.82   558.4  2214.5   579.6 2231.77   594.5 2245.24   598.6 2246.62
     647 2252.84   667.2 2252.56   683.4 2256.97   695.5  2258.9   737.6 2261.22
#Mann= 6 ,-1,0
       0      .1       0      20     .06       0  228.54      .1       0
   261.1    .045       0  355.49     .06       0  428.54      .1       0
#XS Ineff= 2 , 0
                        397.8747            2225
Permanent Ineff=
       F       F
Bank Sta=261.1,355.49
XS Rating Curve= 0 ,0
Exp/Cntr=0.3,0.1

Type RM Length L Ch R = 1 ,30953   ,512.8,512.8,512.8
XS GIS Cut Line= 3
2394338.43957172      714966.378 2394445.7729711714928.957372797
2394760.07151621714306.123060778
#Sta/Elev= 30
       0 2256.87      23 2240.24    44.2 2216.76    52.7 2210.01    61.1 2208.51
     112 2210.36   145.6 2209.34   162.9 2206.16   201.6 2209.14   249.3 2209.05
   261.3 2211.02   276.1 2207.81   297.1  2209.1   359.8 2206.27   413.6 2211.86
   431.5 2211.34     445 2207.96   475.6 2208.19   530.1 2206.62     556 2208.15
   570.4 2214.27   616.2 2217.32   624.2 2216.03   637.6 2208.63   646.6 2207.16
   682.4 2206.87   728.7 2209.97   749.4 2214.94     776 2234.46   811.3 2236.52
#Mann= 6 ,-1,0
       0      .1       0      10     .06       0     110      .1       0
   475.6    .045       0     556     .06       0  623.67      .1       0
#XS Ineff= 2 , 0
                        599.3875            2225
Permanent Ineff=
       F       F
Bank Sta=475.6,556
XS Rating Curve= 0 ,0
Exp/Cntr=0.3,0.1

Type RM Length L Ch R = 1 ,30440   ,546.4,546.4,546.4
XS GIS Cut Line= 2
2394375.85288997715174.2661165832395260.00426299714829.272217707
#Sta/Elev= 30
       0 2268.69    26.1 2250.69    60.5 2217.89    72.1 2210.41    99.1 2206.97
   180.7 2206.15   206.4 2207.91   285.2 2204.23   318.1 2205.69   343.8 2201.84
     361 2202.23   369.6 2205.64   433.5 2207.16   445.8 2211.76   464.1 2204.86
   502.7 2206.59   535.9 2205.16   554.2    2203   610.1 2202.66  650.732205.138
   678.8 2210.78   711.5 2212.28   734.6 2214.17   754.7 2206.24   810.3 2207.92
   846.2 2211.57   862.8 2219.38     902 2245.37   919.2 2251.55   949.1  2256.5
#Mann= 7 ,-1,0
       0      .1       0    72.1     .06       0   180.7      .1       0
   535.9    .045       0  650.73      .1       0   711.5     .06       0
   810.3      .1       0
#XS Ineff= 2 , 0
                           734.6            2215
Permanent Ineff=
       F       F
Bank Sta=535.9,650.73
XS Rating Curve= 0 ,0
Exp/Cntr=0.3,0.1

Type RM Length L Ch R = 1 ,29893   ,336.6,336.6,336.6
XS GIS Cut Line= 3
2394350.29575652715500.4150065712394965.27856222715473.955141741
2395243.73371636715419.588686792
#Sta/Elev= 30
       0 2260.06    41.9 2239.76    61.9 2227.09    73.9 2221.81      98 2207.26
     110 2203.19   242.1 2202.56   294.2 2204.15   342.2 2202.54   378.2 2205.18
   382.2 2204.73   390.2 2199.77   394.2 2199.09   410.3 2201.46   430.3  2201.8
   438.7 2200.16   446.3 2198.31   462.3 2198.07   534.1 2198.58  547.26 2200.17
   562.4 2201.53   582.4 2200.23   598.4 2206.23   724.4 2205.87   740.8 2210.18
   769.3 2210.11   781.5 2207.56   826.4 2207.89   850.8 2211.92   899.3 2216.78
#Mann= 8 ,-1,0
       0      .1       0      90     .06       0     190      .1       0
     290     .05       0   438.7    .045       0  547.26      .1       0
  785.55     .06       0  885.55      .1       0
Bank Sta=438.7,547.26
XS Rating Curve= 0 ,0
Exp/Cntr=0.3,0.1

Type RM Length L Ch R = 1 ,29557   ,648.5,648.5,648.5
XS GIS Cut Line= 4
 2394210.3551232715730.783801477 2394377.6065651715830.525116782
2395157.68758808715799.7398903472395354.01580784715887.598080039
#Sta/Elev= 30
       0 2303.75    14.7 2292.71    48.7 2271.54    99.9 2247.28     111 2239.96
   137.2 2233.85   217.3 2200.91   250.2 2200.95   297.4 2197.91   397.5 2201.61
   549.6 2202.01   597.6  2201.5  603.95 2197.94   609.6 2195.82   689.7 2197.03
   721.7 2195.04   736.1 2197.95   745.7 2201.51   757.7  2202.8   877.8 2204.41
   897.8 2207.54   929.9  2209.1   941.9 2205.85   978.1 2216.22  1065.8 2228.67
  1105.2 2239.35  1127.1  2247.1  1144.9 2255.97  1157.8  2258.9  1190.5 2277.96
#Mann= 8 ,-1,0
       0      .1       0     160     .06       0  264.73     .05       0
  554.73      .1       0  603.95    .045       0   736.1      .1       0
  854.73     .06       0 1055.42      .1       0
Bank Sta=603.95,736.1
XS Rating Curve= 0 ,0
Exp/Cntr=0.3,0.1

Type RM Length L Ch R = 1 ,28908   ,478.1,478.1,478.1
XS GIS Cut Line= 2
2394212.05473081716035.8104985812394925.64078794 716541.92078146
#Sta/Elev= 30
       0 2244.04    78.6 2214.08   110.1 2204.32   124.4 2197.08     211 2195.69
   273.6 2197.44   362.6 2195.44     420 2198.23   500.7 2196.38     520 2197.46
   529.8 2198.13   544.5 2194.85   564.1 2195.92   573.9 2194.58     618  2197.2
   643.7 2196.08   659.2 2193.72   691.6 2191.52   730.8 2191.83   735.7 2192.14
  739.52 2193.73   744.2 2197.88   755.6 2214.59   765.2 2217.63   770.1 2218.57
   799.5 2218.75   804.4 2220.99   814.2  2229.5   818.7 2231.16   874.8 2233.72
#Mann= 9 ,-1,0
       0      .1       0      40     .06       0     210      .1       0
     280     .05       0     520      .1       0     640     .06       0
   659.2    .045       0  739.52     .08       0     760     .05       0
Bank Sta=659.2,739.52
XS Rating Curve= 0 ,0
Exp/Cntr=0.3,0.1

Type RM Length L Ch R = 1 ,28430   ,864.9,864.9,864.9
XS GIS Cut Line= 2
2394011.42858832716395.7964087352394697.41765982716982.167922731
#Sta/Elev= 30
       0 2210.33    45.2  2195.5   100.6 2191.82   151.9 2194.29   191.6 2193.98
   229.9 2191.78   285.1 2193.81   334.6 2192.59   370.3 2193.93   415.7 2193.17
   451.5 2194.88   463.8 2192.76   479.8 2192.74   486.7 2190.12   490.4 2188.76
   500.8 2188.31   585.1 2188.51  598.05 2190.16   611.6 2195.97   648.4 2198.27
   669.3 2201.77   727.8 2217.88   733.5 2218.18   742.9  2215.7   774.5 2215.95
   790.3 2228.47   798.7 2230.64   835.6 2233.03   869.7 2233.74   902.4 2237.03
#Mann= 7 ,-1,0
       0      .1       0      50     .06       0     180     .05       0
   486.7    .045       0  598.05      .1       0     700     .06       0
     850     .05       0
Bank Sta=486.7,598.05
XS Rating Curve= 0 ,0
Exp/Cntr=0.3,0.1

Type RM Length L Ch R = 1 ,27565   ,256.8,256.8,256.8
XS GIS Cut Line= 3
2393361.98928592717051.4990827692394197.09419939717489.723962544
2394393.77047085717533.252266151
#Sta/Elev= 30
       0 2211.19    26.6 2194.36    35.5 2190.51    43.1  2189.2      71 2190.78
   187.7 2189.52   261.9 2190.91   293.2  2185.6   305.1 2187.44   350.3 2188.49
   355.4 2188.25  360.84 2185.33   364.3 2184.01   386.4 2183.73   440.6 2183.81
  464.22 2185.37   490.3 2190.74   512.4 2186.63   815.6 2185.94   835.4 2182.66
   865.3 2185.31   878.8  2189.1   896.9 2197.86   927.2 2202.23   942.2 2195.91
   983.1 2194.01   987.2 2195.02    1019 2216.05  1134.7 2240.98  1144.5 2244.67
#Mann= 7 ,-1,0
       0     .06       0     110      .1       0  360.84    .045       0
  464.22      .1       0     550     .05       0     890     .06       0
  1093.1      .1       0
Bank Sta=360.84,464.22
XS Rating Curve= 0 ,0
Exp/Cntr=0.3,0.1

Type RM Length L Ch R = 1 ,27309   ,505.5,505.5,505.5
XS GIS Cut Line= 3
2393187.49351837717212.8270441352394116.34312876717784.207658168
2394426.87981992 717862.62594858
#Sta/Elev= 30
       0 2229.99    85.3 2206.77   155.8 2197.32   169.9 2189.49   179.3 2187.24
   271.2 2188.33   361.3 2184.19   385.9 2184.41     400 2187.07  412.12 2183.15
   419.4 2180.99   503.3 2181.36  510.94 2183.15   519.8 2188.94   550.3 2184.22
     771 2184.78  1038.9 2181.85  1074.8 2189.23  1098.6 2188.49  1114.2 2182.57
  1135.7 2180.92    1177 2181.78  1185.2 2183.96  1214.1 2202.79  1265.6 2220.52
  1317.3 2243.63  1333.8  2245.4    1342 2250.66  1367.9    2259  1410.8  2279.3
#Mann= 8 ,-1,0
       0      .1       0     200     .06       0     320      .1       0
  412.12    .045       0  510.94      .1       0     610     .05       0
    1010     .06       0 1120.52      .1       0
#XS Ineff= 2 , 0
         254.268    21951069.678            2195
Permanent Ineff=
       F       F
Bank Sta=412.12,510.94
XS Rating Curve= 0 ,0
Exp/Cntr=0.3,0.1

Type RM Length L Ch R = 1 ,26803   ,524.2,524.2,524.2
XS GIS Cut Line= 3
2393198.83366327717949.693216197  2394064.109799 717904.84008421
2394409.20478391718027.589995629
#Sta/Elev= 30
       0 2209.96   197.6 2206.43   221.6  2201.9   233.7  2187.4   249.7 2185.66
  259.85 2179.96   265.7 2177.29   281.7 2177.25   313.8 2177.34  320.63 2180.04
   329.8  2185.8   333.8 2185.93   397.9 2181.97   618.2 2183.09   642.2 2181.13
   678.3  2183.5   830.5 2181.43   850.5 2188.09   866.5 2188.25   883.5 2187.78
   901.2 2181.13  1002.4 2179.98  1023.6 2186.77  1042.1 2200.77  1076.6 2217.97
  1112.7 2242.18  1125.5 2244.02  1138.2 2253.35  1210.4 2274.52  1232.7 2284.77
#Mann= 7 ,-1,0
       0     .05       0     160     .07       0  259.85    .045       0
  320.63      .1       0     360     .05       0     750     .06       0
  956.44      .1       0
#XS Ineff= 2 , 0
                        856.1115            2185
Permanent Ineff=
       F       F
Bank Sta=259.85,320.63
XS Rating Curve= 0 ,0
Exp/Cntr=0.3,0.1

Type RM Length L Ch R = 1 ,26279   ,945.5,945.5,945.5
XS GIS Cut Line= 4
2393197.97768679718345.1607580932393317.11237771718464.354339102
 2393877.3526997718446.9507040712394044.74623972718600.517183513
#Sta/Elev= 30
       0 2202.33    58.1 2203.01   130.1 2197.97   162.8 2188.15   180.8 2181.08
   223.6 2181.25   259.6 2179.15   307.7 2180.49  316.692178.619   319.7 2177.28
   333.6 2176.87   420.4 2176.95   443.7 2178.62   459.7 2182.25   483.7 2179.37
   659.8 2179.09   703.8 2184.07   723.9 2184.48   743.7 2183.74   765.4 2178.75
   831.7 2176.41   840.2 2176.64   845.9  2179.1     874 2206.22     912 2226.54
   922.9 2237.59     928 2239.61   939.1 2240.31     950  2249.5   956.2 2252.67
#Mann= 9 ,-1,0
       0     .05       0     110     .06       0  208.52     .07       0
  308.52      .1       0  316.69    .045       0   443.7      .1       0
  508.52     .05       0  608.52     .06       0  829.03      .1       0
#XS Ineff= 1 ,-1
 721.745 956.198    2185
Permanent Ineff=
       F
Bank Sta=316.69,443.7
XS Rating Curve= 0 ,0
Exp/Cntr=0.3,0.1

Type RM Length L Ch R = 1 ,25333   ,632.7,632.7,632.7
XS GIS Cut Line= 2
2392976.50293103718715.8327385482393447.63116586719435.855174002
#Sta/Elev= 30
       0 2202.47    18.1 2200.21    30.3 2196.86    68.5 2181.61    96.1 2177.15
   361.9 2176.89   408.2 2178.18   417.5 2177.02   448.6 2176.93   460.2  2173.7
   468.8    2170   474.3 2169.22   484.4 2169.03   508.3 2173.53   517.9 2174.03
     537 2171.23   583.8 2173.23  592.49 2171.38   598.5 2169.15   620.4 2167.74
   671.1 2170.69   680.4 2169.31   713.9 2169.54   722.6 2171.45     726 2174.53
   743.3 2195.92   760.7 2210.19     776 2219.65   788.4 2222.77   860.5  2228.5
#Mann= 6 ,-1,0
       0     .05       0     340     .07       0     360     .06       0
     520      .1       0  592.49    .045       0   722.6      .1       0
Bank Sta=592.49,722.6
XS Rating Curve= 0 ,0
Exp/Cntr=0.3,0.1

Type RM Length L Ch R = 1 ,24701   ,429.6,429.6,429.6
XS GIS Cut Line= 3
 2392467.1142712719082.2462758182392908.84348459719769.785782574
2393013.71277011719835.422396772
#Sta/Elev= 30
       0 2203.09    36.8 2196.75    65.3 2188.23    93.8 2181.39   115.8 2178.21
   131.9  2177.3   141.8 2172.86   155.6  2170.9   162.1 2170.77   179.4 2173.43
   283.2 2171.47   355.3 2173.53   457.4 2171.81     574  2174.3   607.3 2172.95
   616.8  2169.9   632.7 2167.82   640.6  2165.5   712.1 2165.38   732.3  2165.7
  739.32 2167.82   745.2 2170.12   756.8 2169.11   773.7 2172.18   808.6 2174.08
     816 2176.33   835.3 2186.31   854.2 2190.01   883.9 2209.19   940.9 2213.82
#Mann= 9 ,-1,0
       0      .1       0      10     .05       0      30      .1       0
     190     .05       0     560     .06       0   632.7    .045       0
  739.32     .06       0     740      .1       0  887.21     .05       0
#XS Ineff= 2 , 0
        197.0334    2180
Permanent Ineff=
       F       F
Bank Sta=632.7,739.32
XS Rating Curve= 0 ,0
Exp/Cntr=0.3,0.1

Type RM Length L Ch R = 1 ,24271   ,377.4,377.4,377.4
XS GIS Cut Line= 4
2392001.97454599 719575.360346392392193.87962415719681.969988884
 2392593.2467072719989.668779555 2392789.5907367 720193.55752018
#Sta/Elev= 30
       0 2265.45    25.4 2252.61    35.3 2249.73    84.9 2222.44   114.7 2210.15
   121.5 2205.52   135.3 2204.28     152 2195.53     200  2176.1   222.4 2169.97
   237.7 2167.54   331.8 2167.54   528.6 2170.93   545.6 2169.68   560.7 2164.87
   571.4 2162.56   631.3 2162.53   646.6 2162.87  653.34 2164.88   665.5 2169.84
   739.4 2169.04   773.5 2164.88   790.5 2165.44   806.3 2169.72   831.7 2169.48
   843.2 2173.28   861.8 2186.99   872.9 2191.52   939.6 2197.02  1006.7 2206.21
#Mann= 7 ,-1,0
       0      .1       0  319.53     .05       0  409.53     .06       0
  449.53     .07       0   560.7    .045       0  653.34      .1       0
 1003.68     .05       0
Bank Sta=560.7,653.34
XS Rating Curve= 0 ,0
Exp/Cntr=0.3,0.1

Type RM Length L Ch R = 1 ,23894   ,506.2,506.2,506.2
XS GIS Cut Line= 2
 2391916.6186108720004.781025857 2392655.3211678720436.516032361
#Sta/Elev= 30
       0 2232.95    32.1 2215.21    46.8  2210.7    64.3 2201.58      69 2198.81
    78.2 2189.59    92.1  2188.1   111.8 2171.66   124.6 2166.57   181.3  2165.6
   201.7 2167.59   240.4 2166.11     384 2168.74   388.9 2168.55   404.6 2163.13
   425.7 2160.81   494.1 2163.13   509.1 2162.88   532.3  2170.6   560.1 2170.67
   573.1 2162.56   578.9 2161.95   606.4 2162.28   620.3 2165.27   643.3 2166.76
     655 2169.56   698.8 2195.62   708.3 2198.88   777.8  2206.6   855.6 2207.82
#Mann= 5 ,-1,0
       0      .1       0     300     .06       0   404.6    .045       0
   494.1      .1       0     760     .05       0
Bank Sta=404.6,494.1
XS Rating Curve= 0 ,0
Exp/Cntr(USF)=0,0
Exp/Cntr=0.3,0.1

Type RM Length L Ch R = 1 ,23387   ,322.5,322.5,322.5
XS GIS Cut Line= 2
2391732.74162094720539.1593663282392494.60961939720804.662134939
#Sta/Elev= 30
       0 2222.39    20.6 2213.97    33.3 2210.71    58.7 2198.67    67.2 2192.99
    84.1 2190.71    95.4  2187.2   109.5  2178.3   122.2 2167.64   129.9 2163.67
   133.1 2162.99   198.5 2163.23   236.6 2165.15   308.6 2163.73   333.9 2162.22
   473.8 2164.36     532 2163.22   545.8 2163.69  557.51  2159.9   571.3 2156.94
     584 2156.38   596.7 2156.75   601.7 2159.88   632.5  2181.8   647.5 2187.83
   664.4 2202.27   668.7 2205.18   677.1    2209   745.6 2203.77   806.8 2201.87
#Mann= 7 ,-1,0
       0      .1       0     160     .06       0     260      .1       0
     370     .05       0  557.51    .045       0   601.7      .1       0
     790     .05       0
Bank Sta=557.51,601.7
XS Rating Curve= 0 ,0
Exp/Cntr=0.3,0.1

Type RM Length L Ch R = 1 ,23065   ,502.9,502.9,502.9
XS GIS Cut Line= 3
2391644.74124719720996.2621148012392098.03424719721035.629114801
2392338.34413061721057.409270313
#Sta/Elev= 30
       0 2210.41     7.5 2209.88    15.5 2207.07    51.6 2185.13    67.7 2182.91
    83.7 2174.66   103.8 2167.37   123.9 2169.28     140 2162.76     148 2159.69
     156 2159.45     160 2159.63   172.1 2164.44   188.7 2161.86   208.2 2161.09
   392.9 2163.93   441.1  2159.6   493.3  2159.5   533.5 2161.61   545.5 2160.67
   550.5 2158.18   557.6 2155.49   617.8  2155.7   624.1 2158.22   625.8 2159.62
   645.9 2190.38     654 2198.52     658 2200.43     666 2201.12   696.3 2199.86
#Mann= 7 ,-1,0
       0     .06       0      40     .07       0     140     .06       0
     340     .05       0     535      .1       0   550.5    .045       0
   624.1      .1       0
Bank Sta=550.5,624.1
XS Rating Curve= 0 ,0
Exp/Cntr=0.3,0.1

Type RM Length L Ch R = 1 ,22562   ,378.9,378.9,378.9
XS GIS Cut Line= 2
2391650.93114031721488.6117849972392364.13483345721562.863128393
#Sta/Elev= 30
       0 2194.04    17.3 2183.47    29.4 2180.58    37.4 2175.17    45.5 2173.19
    73.6 2162.34    85.7 2159.06   109.8 2157.73   113.9 2155.78   117.9 2154.86
   129.9 2158.41   150.1  2159.3   218.4 2157.98   351.1 2160.43   427.8 2158.41
   447.7 2158.75   471.8  2160.7   495.9 2159.75   511.6 2156.31     516 2153.66
   528.1 2153.76   548.2 2151.65   560.3 2151.25   600.5 2152.26   604.5 2153.02
  609.57  2155.9   620.2 2166.24   624.6 2168.07   660.9 2168.88717.0584  2167.9
#Mann= 7 ,-1,0
       0      .1       0      40     .05       0     140     .06       0
     230     .05       0   511.6    .045       0  609.57     .05       0
     630      .1       0
Bank Sta=511.6,609.57
XS Rating Curve= 0 ,0
Exp/Cntr(USF)=0,0
Exp/Cntr=0.3,0.1

Type RM Length L Ch R = 1 ,22183   ,274.1,274.1,274.1
XS GIS Cut Line= 2
2391719.36507786721867.7622202572392348.30733267721912.387118768
#Sta/Elev= 30
       0 2196.42     8.8 2195.13    25.2  2186.6    44.9  2178.2      61 2172.61
      85 2165.94   125.1  2159.2   141.2 2158.47   149.2 2155.86   165.2 2152.33
   170.6 2152.42   181.3 2155.32   189.3 2155.94   265.5 2156.26   285.5 2157.04
   301.6  2156.5   313.6 2158.56   320.4 2157.59   327.8 2154.81   333.6  2151.5
   337.7 2150.85  399.542154.869   413.8 2156.13   429.9 2159.49   445.9 2171.63
   449.9  2173.9   453.9 2174.87   570.2 2181.26   590.7 2181.78   630.5 2180.95
#Mann= 3 ,-1,0
       0      .1       0   327.8    .045       0  399.54      .1       0
Bank Sta=327.8,399.54
XS Rating Curve= 0 ,0
Exp/Cntr=0.3,0.1

Type RM Length L Ch R = 1 ,21909   ,423.8,423.8,423.8
XS GIS Cut Line= 2
2391790.10675591722281.1126716982392341.19826356722056.668049652
#Sta/Elev= 30
       0 2237.37    10.7 2231.28    41.1 2216.06    49.7 2212.09    58.4 2209.26
    88.6  2194.2    97.3 2187.62   118.2 2167.87   124.3 2160.65   127.5  2158.2
   153.4 2156.47     270 2155.19   274.7 2154.84  284.032151.462   291.6  2149.5
   339.1 2149.28   357.5 2150.84   386.6  2150.2   399.6 2149.04   403.9 2149.26
  411.442151.461   418.9 2154.25   421.2 2155.55   425.5 2159.74   437.3 2165.86
   451.4 2171.03   458.8 2172.67   520.5 2178.26   551.3 2180.18     595 2180.63
#Mann= 3 ,-1,0
       0      .1       0  284.03    .045       0  411.44      .1       0
Bank Sta=284.03,411.44
XS Rating Curve= 0 ,0
Exp/Cntr=0.3,0.1

Type RM Length L Ch R = 1 ,21485   ,540.2,540.2,540.2
XS GIS Cut Line= 3
2392291.60416231722683.1633672432392416.25316231722257.729367243
2392366.29711703722149.677659177
#Sta/Elev= 30
       0 2270.49    18.2  2255.4    35.4 2239.34    56.3 2221.36    69.8 2207.64
      73 2204.07    77.1 2197.96    81.3 2188.52    85.4 2181.65    89.6 2177.43
    93.8  2171.6    97.9 2164.26   102.1 2158.16   106.3 2156.54   131.3 2154.88
   181.3 2155.04   185.5 2154.26  193.192149.674     198 2147.44   202.1 2146.97
   264.7 2145.61   302.2 2147.06     315 2149.72   331.4 2148.25   350.2  2153.1
   398.6  2155.5   417.9 2157.68   435.6 2157.72   496.8 2168.56   562.4 2176.72
#Mann= 3 ,-1,0
       0      .1       0  193.19    .045       0     315      .1       0
Bank Sta=193.19,315
XS Rating Curve= 0 ,0
Exp/Cntr=0.3,0.1

Type RM Length L Ch R = 1 ,20945   ,656.9,656.9,656.9
XS GIS Cut Line= 3
2392807.73850524722791.7067020222392930.65355066722370.624170257
2393490.14137303722330.589068589
#Sta/Elev= 30
       0 2288.79    19.3 2276.91    30.1 2263.23    65.1 2226.34    73.5 2212.79
    77.6 2202.18    81.8 2196.53      86  2186.8    90.1 2171.66    94.3  2165.8
   119.3 2153.27   144.3 2152.84  158.67 2146.61   244.3 2144.75   290.2 2146.66
   306.8 2144.79   331.8 2146.92     361 2145.29     411 2153.58   488.3 2151.56
     765 2151.32   833.2 2151.76   877.3 2154.58   893.3 2150.17   946.7 2149.15
   961.5 2151.21   969.5 2154.69   985.6 2178.85   993.6  2184.2   999.6 2185.84
#Mann= 3 ,-1,0
       0      .1       0  158.67    .045       0   290.2      .1       0
Bank Sta=158.67,290.2
XS Rating Curve= 0 ,0
Exp/Cntr=0.3,0.1

Type RM Length L Ch R = 1 ,20288   ,355,355,355
XS GIS Cut Line= 4
2393166.79165808723090.6179057412393451.45636328722888.295564711
2393522.75205242722696.1932911752393728.76601871722548.589260421
#Sta/Elev= 30
       0 2247.53    50.8    2208    55.7  2202.6    60.6 2190.99    65.5 2183.63
    73.7    2176    93.8 2160.88   104.8 2150.49   109.7 2147.96   131.1 2147.97
   154.1 2141.14   163.6  2141.9   174.1 2146.99   188.5 2146.55   237.2 2148.91
   260.2 2148.52   278.7  2145.4   340.5 2145.06   356.8 2142.97   380.4 2142.38
   403.8 2141.21   506.2 2140.92   531.8 2142.37   551.4 2147.62   573.1 2150.15
   597.5 2156.03   621.1 2159.05   724.2 2162.52   763.7 2166.11   807.6 2167.39
#Mann= 3 ,-1,0
       0      .1       0   380.4    .045       0   531.8      .1       0
Bank Sta=380.4,531.8
XS Rating Curve= 0 ,0
Exp/Cntr=0.3,0.1

Type RM Length L Ch R = 1 ,19933   ,513.9,513.9,513.9
XS GIS Cut Line= 3
2393459.58920879723477.3405325072393588.30856029723364.441396819
     2394029.746      722500.575
#Sta/Elev= 30
       0    2248    80.6  2199.7   127.6 2162.76   139.1 2147.87   144.4 2144.01
   167.8 2143.36   179.7 2137.37   192.8 2135.14   221.1 2141.96   301.4 2145.25
   320.4 2141.14   346.7 2146.36   375.7 2143.87   439.9 2147.44   471.4 2141.91
   509.5 2145.08   543.2 2142.58     651  2141.3   664.5  2138.4   693.4 2138.14
   717.6 2138.37   724.5 2141.32   740.9  2149.5   754.3  2152.2   900.5 2160.87
   919.7 2165.89   965.5 2163.87  1046.3  2173.9  1104.7 2176.37  1141.3 2181.48
#Mann= 3 ,-1,0
       0      .1       0     651    .045       0   724.5      .1       0
Bank Sta=651,724.5
XS Rating Curve= 0 ,0
Exp/Cntr=0.3,0.1

Type RM Length L Ch R = 1 ,19419   ,524.3,524.3,524.3
XS GIS Cut Line= 3
2393636.94057189723646.993509308 2394344.2678608723096.796104397
2394486.85267979722804.683421095
#Sta/Elev= 30
       0 2233.22    80.1 2174.11    90.2 2155.97   100.5 2144.99   120.7 2142.53
   135.9 2133.75   166.3 2134.25   176.4 2140.66   181.5 2141.39   231.6 2142.12
     243 2138.19   252.4 2137.84   272.7 2140.51   318.3 2139.18   404.4  2143.3
   442.6 2142.81   470.3 2139.78   530.9 2145.97   630.7 2144.58   662.9 2137.84
   688.2 2140.78   706.6 2140.29   804.3 2137.97  842.822140.242   852.1 2145.71
   869.4 2149.36  1078.1 2158.77    1141 2165.72    1185 2165.44  1221.2 2174.48
#Mann= 3 ,-1,0
       0      .1       0   706.6    .045       0  842.82      .1       0
Bank Sta=706.6,842.82
XS Rating Curve= 0 ,0
Exp/Cntr=0.3,0.1

Type RM Length L Ch R = 1 ,18895   ,262,262,262
XS GIS Cut Line= 4
2393762.19938279723900.7960615062393862.10174717723804.081759095
2394788.71760561723535.483845697  2394973.556884  723384.5727529
#Sta/Elev= 30
       0 2234.47    60.5 2194.31     103 2172.28   130.8 2143.37   152.7 2142.48
   174.5 2138.01   224.5 2137.59   249.3 2132.14   266.1 2136.92   282.8 2138.53
   357.8 2138.73   375.5 2134.92   386.9 2134.44   399.4 2135.48   411.9 2139.13
   474.4 2138.21   682.3 2141.04   695.2 2136.47  738.37 2137.81     796 2136.09
   836.7 2136.28   847.5 2137.83   857.5 2141.44   932.5 2136.67  1011.6 2136.72
  1024.1 2143.51  1032.4 2145.31  1094.9 2152.59  1244.4 2158.57  1342.4 2165.53
#Mann= 3 ,-1,0
       0      .1       0  738.37    .045       0   847.5      .1       0
Bank Sta=738.37,847.5
XS Rating Curve= 0 ,0
Exp/Cntr=0.3,0.1

Type RM Length L Ch R = 1 ,18633   ,739.2,739.2,739.2
XS GIS Cut Line= 4
2393892.03435686724084.0084589712394423.40871543723871.568461587
2394578.32433897723882.4743411562395112.99365586 723650.00441105
#Sta/Elev= 30
       0 2202.62    45.4 2178.46    77.7 2158.61      82 2155.48    90.6 2142.11
   107.8 2141.63   125.1 2131.68   168.2 2129.62   202.6 2130.23   215.5  2133.4
   228.5 2134.09   330.9 2134.95   357.7 2133.45     418 2136.25   605.1 2135.85
  719.77 2135.91   729.6  2137.5     795 2138.61   812.5 2133.84   842.4  2133.6
   873.5 2136.01   901.4 2133.59   948.8 2134.02   960.8 2134.74   973.8 2140.46
    1000 2142.57  1034.9 2143.12  1126.5 2150.09    1238 2155.12  1310.6 2161.92
#Mann= 3 ,-1,0
       0      .1       0   605.1    .045       0  719.77      .1       0
Bank Sta=605.1,719.77
XS Rating Curve= 0 ,0
Exp/Cntr=0.3,0.1

Type RM Length L Ch R = 1 ,17894   ,544,544,544
XS GIS Cut Line= 3
2394057.42532699724668.998240793   2394915.63216724357.929214593
2395307.67867541724279.163378334
#Sta/Elev= 30
       0  2242.3    19.9 2211.54   108.2  2145.2   122.1 2137.23   143.3 2136.94
   156.1 2128.83   173.8 2125.75   249.7  2133.8     271 2134.76   279.9 2132.08
     288 2129.98   351.8 2129.53  378.19 2132.11   458.2 2133.41   475.2  2130.7
   492.2 2132.04   513.5    2129   547.5 2131.61   666.7 2130.66   683.7 2132.56
   696.4 2136.12   734.7 2136.69     995 2137.74  1007.2 2135.59  1068.4 2136.11
  1084.8 2137.32  1117.4 2145.56  1168.7 2153.13  1215.3 2156.68  1312.7 2170.75
#Mann= 3 ,-1,0
       0      .1       0   279.9    .045       0  378.19      .1       0
Bank Sta=279.9,378.19
XS Rating Curve= 0 ,0
Exp/Cntr=0.3,0.1

Type RM Length L Ch R = 1 ,17350   ,491.6,491.6,491.6
XS GIS Cut Line= 4
2394065.13875815725147.1787597412394521.50294114725082.936721393
2394685.87911334724997.7779815782395503.78448149 724891.87021488
#Sta/Elev= 30
       0 2235.01       8 2227.93    31.3 2197.93    62.3 2165.67     100 2131.79
   108.1 2127.48   148.5 2127.09   184.8 2131.15   261.6 2132.39   273.7 2132.03
   289.9 2125.82   358.6 2126.75   398.9 2130.15   439.3 2128.97   463.9 2131.55
   482.1 2128.05   493.8 2125.53     572 2125.15  634.78 2128.03   664.4 2131.24
     733 2128.24   753.2 2132.58     971 2130.46  1030.7 2132.92    1102 2132.11
  1128.3 2135.61  1152.5 2141.52  1253.3 2154.69  1414.6 2172.86  1470.7 2177.18
#Mann= 3 ,0,0
       0      .1       0   482.1    .045       0  634.78      .1       0
Bank Sta=482.1,634.78
XS Rating Curve= 0 ,0
Exp/Cntr=0.3,0.1

Type RM Length L Ch R = 1 ,16858   ,1016.7,1016.7,1016.7
XS GIS Cut Line= 2
 2394167.8749798725571.3072816972395442.85009957725451.570296533
#Sta/Elev= 30
       0  2232.1     8.3    2221    20.4 2210.36    24.4 2204.21    32.4  2186.2
    40.5  2175.6      94 2128.05    96.7 2126.46   130.8 2123.99     153  2125.1
   177.1 2119.88   269.5 2122.25   325.4 2129.34   341.8 2122.87   353.9 2121.97
   414.8 2127.95   438.2 2125.75   474.4 2127.51   490.1 2124.64   498.5 2122.15
   534.5 2121.72   594.9 2122.26  604.02 2124.64   631.1  2129.1   707.4 2130.81
   823.9 2127.53   908.3 2128.08   971.8 2136.21  1126.1  2151.1  1280.6 2175.02
#Mann= 3 ,-1,0
       0      .1       0   490.1    .045       0  604.02      .1       0
Bank Sta=490.1,604.02
XS Rating Curve= 0 ,0
Exp/Cntr=0.3,0.1

Type RM Length L Ch R = 1 ,15841   ,899.6,899.6,899.6
XS GIS Cut Line= 3
2394098.74604451725916.2504100332394231.04261883726355.085880496
2394997.58735797      726585.809
#Sta/Elev= 30
       0 2174.32    46.9 2145.16    85.4 2124.88   109.6 2124.31   122.1 2121.27
   201.5 2121.01     217 2117.71   251.6 2117.63   306.8    2119   318.5 2121.72
   467.4 2121.99   522.2 2124.35   595.8 2123.53   630.8 2120.12   714.3 2124.49
   724.2 2122.81   737.1 2117.65   756.3 2120.92   810.9 2122.96   835.5  2122.4
   955.4 2124.59  966.55 2121.48   985.9  2118.3  1102.8 2118.89 1113.382121.466
  1115.4 2122.38  1136.2 2144.59  1141.6 2148.98  1148.8 2152.38  1258.9 2162.28
#Mann= 3 ,0,0
       0      .1       0  966.55    .045       0 1113.38      .1       0
Bank Sta=966.55,1113.38
XS Rating Curve= 0 ,0
Exp/Cntr=0.3,0.1

Type RM Length L Ch R = 1 ,14942   ,543.6,543.6,543.6
XS GIS Cut Line= 2
2393918.52686824725812.9070402542394246.52402925 727285.44083072
#Sta/Elev= 30
       0 2240.36      29 2235.53    49.5 2228.55    82.2  2208.9   139.6 2167.43
   176.5 2143.99   205.2 2129.24   226.2 2124.24   311.7 2120.73   332.2 2116.44
   377.3 2120.01   410.1 2116.51   528.9 2116.55   559.5  2119.9   695.4 2119.41
   758.4 2121.93   919.9 2118.22   943.4 2115.08  1181.3 2117.81  1203.4 2114.76
  1295.3 2117.25 1306.66 2114.32  1315.7 2111.67  1373.1 2111.36  1426.4 2112.03
 1435.23 2114.32  1442.8 2123.94  1459.5 2138.71  1483.8 2150.69  1508.6 2171.85
#Mann= 3 ,-1,0
       0      .1       0 1306.66    .045       0 1435.23      .1       0
Bank Sta=1306.66,1435.23
XS Rating Curve= 0 ,0
Exp/Cntr(USF)=0,0
Exp/Cntr=0.3,0.1

Type RM Length L Ch R = 1 ,14398   ,494.5,494.5,494.5
XS GIS Cut Line= 4
2393491.83842214726133.133076096 2393530.0488501726209.781990415
2393698.71837465727364.372049289 2393752.8836637727456.795305855
#Sta/Elev= 30
       0 2157.17    59.9 2124.99    80.5 2124.35   101.1 2118.32   113.3 2116.81
   202.3 2117.47   226.5 2115.41   254.8 2115.47   263.3 2110.87     275 2109.71
   316.3 2115.18   339.7 2112.74   392.3 2115.87     655 2117.78   787.8 2114.83
     934  2113.9   970.3 2113.06   986.4 2111.19  1010.8 2111.72  1051.2 2108.68
  1081.3 2108.72  1095.7 2105.56  1140.1 2105.55  1192.7 2105.66 1206.54 2108.72
  1255.4 2116.02  1268.8 2121.62  1279.1 2123.42  1318.3 2146.52  1359.6 2164.45
#Mann= 3 ,-1,0
       0      .1       0  1081.3    .045       0 1206.54      .1       0
Bank Sta=1081.3,1206.54
XS Rating Curve= 0 ,0
Exp/Cntr=0.3,0.1

Type RM Length L Ch R = 1 ,13904   ,677.5,677.5,677.5
XS GIS Cut Line= 3
2393061.00752116726580.0326406142393131.03803643726789.198605811
2393212.69555169727497.048269429
#Sta/Elev= 30
       0 2130.13    43.4 2127.67    51.8 2124.46    60.3 2119.56    72.9 2107.59
    81.4 2105.78   110.9 2105.91   169.9 2109.55   225.2 2111.02   329.3 2112.08
   459.9 2111.54   534.6 2109.22   570.9 2111.67     587 2109.88   603.1 2104.28
   615.2 2105.35   631.3 2108.77   680.1 2108.01   695.7  2107.1   701.7 2105.22
   711.8  2101.4   783.7    2101   804.4  2102.3  810.59 2105.27   816.5 2109.84
   824.5 2119.08   872.9 2157.26   892.9 2177.06   905.1 2184.64   933.1 2204.38
#Mann= 3 ,-1,0
       0      .1       0   701.7    .045       0  810.59      .1       0
Bank Sta=701.7,810.59
XS Rating Curve= 0 ,0
Exp/Cntr=0.3,0.1

Type RM Length L Ch R = 1 ,13226   ,537.7,537.7,537.7
XS GIS Cut Line= 3
 2392882.2620932726475.3600583982392793.33815425726719.933502433
2392506.74144831727184.613971096
#Sta/Elev= 30
       0 2131.49      70 2128.87    90.4 2127.14   193.5 2126.19   227.8 2124.25
   240.3 2121.91   270.7 2111.25   299.3 2106.54   318.1 2107.14     398 2105.01
   421.5 2105.47   430.1 2107.44   454.4 2107.98   477.9 2107.56     492 2105.41
   520.7 2105.56   543.7 2108.93   549.8 2108.96   562.5 2106.86  606.922103.499
   618.9 2100.62   657.3 2100.53   717.6 2100.77  723.322103.495     730 2108.77
   742.5 2121.59   764.6 2139.88     774 2146.53   799.7 2167.31   806.2 2171.36
#Mann= 3 ,-1,0
       0      .1       0  606.92    .045       0  723.32      .1       0
Bank Sta=606.92,723.32
XS Rating Curve= 0 ,0
Exp/Cntr=0.3,0.1

Type RM Length L Ch R = 1 ,12689   ,381.5,381.5,381.5
XS GIS Cut Line= 3
2392611.73206095726196.9917562232392318.67906095726545.051756223
2392025.62706095726893.110756223
#Sta/Elev= 30
       0 2136.42    86.3 2129.87   138.9 2123.93   161.6 2120.04   192.9 2116.76
   235.5 2110.36   258.2 2108.58   277.4 2106.05   287.8 2106.98   328.5 2107.34
   502.4 2106.28   533.6 2102.82   549.3 2099.64   585.9 2101.28   618.7 2101.03
   644.2    2102   652.7    2101   666.9 2098.56   674.8 2098.05   729.4 2097.97
   758.4 2099.05   789.8 2098.17   800.3 2096.91     816 2097.11   821.2 2098.46
   825.9  2101.1   831.7 2106.24   845.8 2121.47   857.1 2132.17     910 2173.61
#Mann= 3 ,-1,0
       0      .1       0   652.7    .045       0   825.9      .1       0
Bank Sta=652.7,825.9
XS Rating Curve= 0 ,0
Exp/Cntr=0.3,0.1

Type RM Length L Ch R = 1 ,12307   ,604.7,604.7,604.7
XS GIS Cut Line= 2
2392221.49741429726061.6701271522391718.82106508726674.846161955
#Sta/Elev= 30
       0 2145.64    33.6 2124.39    51.1 2115.77    65.2 2110.72    82.1 2107.66
   100.1 2106.54   144.2 2106.04   154.5 2103.88   165.4 2103.15   202.4 2104.98
   267.8 2104.52   330.4 2102.97   378.6 2105.33   412.2 2105.51   478.1 2102.47
   487.9 2100.59   500.5 2097.81   506.8 2097.85     515 2096.74   526.4 2097.54
   540.6  2096.9   677.2 2096.94   682.7 2097.46  688.23 2100.63   697.6 2107.73
   708.7 2118.51   733.8 2137.51   748.1 2147.63   779.4 2165.52   792.9 2173.93
#Mann= 3 ,0,0
       0      .1       0   487.9    .045       0  688.23      .1       0
Bank Sta=487.9,688.23
XS Rating Curve= 0 ,0
Exp/Cntr=0.3,0.1

Type RM Length L Ch R = 1 ,11702   ,638.6,638.6,638.6
XS GIS Cut Line= 4
 2392092.8093647725743.4664281492391922.89609919725922.677935862
 2391786.9036057725939.4578249612391394.30789276726481.002456115
#Sta/Elev= 30
       0 2180.98    46.5 2178.92    63.9 2175.85    88.1  2165.8   156.7 2123.34
   178.7 2113.01   199.7  2107.1   253.7 2104.07   268.52095.469   277.9 2092.55
   326.3 2092.03   370.6 2093.56     379 2095.41   400.9 2098.54   436.3 2099.96
   554.1 2099.69   583.7 2101.88   652.9 2102.52   733.7 2099.26     743 2100.42
   761.6 2098.14   790.7 2100.97   811.2 2098.84   868.3 2100.27   908.4 2096.42
   939.4 2100.53   954.3  2105.5  1020.1 2146.11  1034.5 2152.01  1052.9 2164.24
#Mann= 3 ,-1,0
       0      .1       0   268.5    .045       0     379      .1       0
Bank Sta=268.5,379
XS Rating Curve= 0 ,0
Exp/Cntr=0.3,0.1

Type RM Length L Ch R = 1 ,11064   ,609.2,609.2,609.2
XS GIS Cut Line= 2
2391495.17541779725220.9340771722391065.39125336726314.526111974
#Sta/Elev= 30
       0  2173.2   107.7 2157.28   120.6 2153.07   167.9 2147.41   209.2 2145.68
   223.7 2138.99   245.2 2133.21   279.6 2120.21   292.5 2112.51  316.68 2092.13
   325.3 2088.09   365.6  2087.9     400 2088.05   412.8 2092.16   442.9 2096.48
   464.4 2097.69   541.8 2096.02   653.5 2099.22   764.6 2098.86   823.2 2100.59
   881.3 2099.52   971.6 2101.57  1036.1 2090.59  1060.8 2090.85    1070 2092.76
    1079 2097.32  1094.7 2100.15  1147.1 2134.45  1156.4 2136.87    1175 2148.47
#Mann= 3 ,-1,0
       0      .1       0  316.68    .045       0   412.8      .1       0
Bank Sta=316.68,412.8
XS Rating Curve= 0 ,0
Exp/Cntr=0.3,0.1

Type RM Length L Ch R = 1 ,10455   ,407,407,407
XS GIS Cut Line= 2
2390873.67834272725061.2350427582390554.62794101726168.543572473
#Sta/Elev= 30
       0 2174.37      82 2164.92   132.2 2156.08   141.5 2152.01   166.5 2151.39
   188.6 2141.09   199.8 2128.34   216.4    2127   220.6 2124.05   246.8 2089.87
     251 2086.88   303.8 2086.69   353.8 2086.77   366.3 2089.87   366.3 2089.89
   391.2 2093.81     462 2087.06     487 2086.97   499.5 2091.99   524.4 2091.96
   549.4 2098.47     641 2094.97   711.8 2097.15   915.8    2096  1007.3 2088.88
  1053.1 2087.94  1061.4 2090.14  1082.3 2103.95  1107.2 2124.21  1152.4 2155.58
#Mann= 3 ,-1,0
       0      .1       0   246.8    .045       0   366.3      .1       0
Bank Sta=246.8,366.3
XS Rating Curve= 0 ,0
Exp/Cntr=0.3,0.1

Type RM Length L Ch R = 1 ,10048   ,1141.1,1141.1,1141.1
XS GIS Cut Line= 2
2390488.38021224724943.2638967822390162.99092929726032.411996931
#Sta/Elev= 30
       0 2146.86    70.6 2134.33   118.9 2122.87   143.1 2124.69   162.4 2118.15
   185.7 2117.58   189.9 2115.64   198.2  2107.7   223.3 2104.93   248.3 2098.66
  268.08 2088.76   290.1 2084.96   353.8 2084.82   381.9 2085.01   402.8 2088.75
     432 2088.84   448.5 2085.67   461.2 2089.62   482.1 2090.92   490.4 2093.85
     528 2092.34   567.4 2095.38   866.2 2091.79   904.9 2086.53   953.8 2088.92
   995.6 2087.56  1012.3 2091.21  1074.9 2091.61  1087.4 2096.36  1136.7 2138.29
#Mann= 3 ,-1,0
       0      .1       0  268.08    .045       0   402.8      .1       0
Bank Sta=268.08,402.8
XS Rating Curve= 0 ,0
Exp/Cntr(USF)=0,0
Exp/Cntr=0.3,0.1

Type RM Length L Ch R = 1 ,8906    ,434.7,434.7,434.7
XS GIS Cut Line= 2
 2389837.7944339724743.8209585942389346.18606946725908.438489996
#Sta/Elev= 30
       0 2137.43    27.5 2137.92    62.3  2131.7   117.3 2131.99   209.9 2125.47
   307.6 2123.48   361.8 2115.35   405.3  2097.5   409.6 2094.05     453 2089.41
   557.2 2087.09   661.4 2090.12   874.2 2088.86   978.4  2085.6  1008.8 2079.87
  1030.5 2076.99  1104.3 2075.14  1144.1 2075.52 1157.52 2079.97  1165.1 2087.18
  1182.4 2091.14  1199.8 2122.13  1205.2 2135.23  1208.5 2146.37  1212.8 2167.07
  1214.3 2169.73  1246.7 2204.49  1257.1 2212.57  1260.6 2217.59  1264.1 2226.06
#Mann= 3 ,-1,0
       0      .1       0  1008.8    .045       0 1157.52      .1       0
Bank Sta=1008.8,1157.52
XS Rating Curve= 0 ,0
Exp/Cntr=0.3,0.1

Type RM Length L Ch R = 1 ,8472    ,352.2,352.2,352.2
XS GIS Cut Line= 3
2389369.45123356724722.4869993872388964.26633148725701.609296722
2388960.10019286725776.748890111
#Sta/Elev= 30
       0 2132.64    11.6  2129.1    33.2 2125.99    67.8 2118.42   119.8 2115.09
   150.1 2111.55   253.7 2095.06     293 2090.87   310.3 2091.28   349.2 2084.05
   486.8 2085.81     544 2084.97   714.7 2086.44   855.7 2085.14   877.4 2086.11
     886 2085.03     903 2079.26   916.3 2074.58  1020.2 2074.16  1024.6  2074.4
 1034.24 2079.06  1041.9 2086.57  1046.2 2088.93  1056.3 2087.21  1066.9 2089.56
  1079.2 2100.39  1087.3 2108.37  1103.3 2128.16  1119.3 2142.57  1134.9 2178.15
#Mann= 3 ,-1,0
       0      .1       0     903    .045       0 1034.24      .1       0
Bank Sta=903,1034.24
XS Rating Curve= 0 ,0
Exp/Cntr=0.3,0.1

Type RM Length L Ch R = 1 ,8120    ,587,587,587
XS GIS Cut Line= 4
2388903.68508345724629.9805937732388902.19596016724849.105962927
2388620.43465121725626.814379498 2388614.9250165725722.997370944
#Sta/Elev= 30
       0 2121.39   111.2 2111.79     249 2097.84   287.3 2093.16   295.8 2090.31
   312.8 2089.76   325.6 2083.12   339.4 2080.93   376.6 2081.28   402.1 2083.68
   492.5 2081.95   567.4 2082.54   612.6 2084.66   738.2 2084.78   779.8  2083.6
   819.1 2084.48   853.1 2083.91   857.4 2082.85   867.2 2076.26   878.6 2073.03
   973.4 2072.44   989.3 2072.79   997.8 2075.54  1010.5 2077.51  1020.2 2083.52
  1031.8 2083.71  1056.7 2087.84  1065.5 2105.79  1105.6  2141.4  1142.6 2172.25
#Mann= 3 ,-1,0
       0      .1       0   867.2    .045       0   997.8      .1       0
Bank Sta=867.2,997.8
XS Rating Curve= 0 ,0
Exp/Cntr=0.3,0.1

Type RM Length L Ch R = 1 ,7533    ,968.3,968.3,968.3
XS GIS Cut Line= 4
2388297.81639121724557.4499320462388309.65575092724689.256116473
2388062.11288981725460.8292881042388050.49844964725563.204771243
#Sta/Elev= 30
       0 2114.64      24 2110.35    68.3 2100.34   157.5 2087.04   195.3 2087.69
   291.9 2081.45   350.7 2082.67   363.3    2080   380.1 2079.68   396.9  2076.8
   451.5 2077.56   472.5 2080.12   524.6 2082.69   590.1 2078.67   702.8 2081.96
   707.8 2081.24  723.26 2075.83   745.6  2072.5   758.2 2072.25     880 2072.34
   884.2 2072.83  892.422075.829   905.2 2081.09   938.8 2082.43     947 2084.32
   951.1 2087.56   959.1 2097.47   998.9 2128.51  1023.5 2145.36  1045.7 2156.79
#Mann= 3 ,-1,0
       0      .1       0  723.26    .045       0  892.42      .1       0
Bank Sta=723.26,892.42
XS Rating Curve= 0 ,0
Exp/Cntr=0.3,0.1

Type RM Length L Ch R = 1 ,6564    ,249.3,249.3,249.3
XS GIS Cut Line= 3
2387629.78093002724514.2495177512387223.20121926725053.270437476
2387105.52452199725408.926491732
#Sta/Elev= 30
       0 2119.54    68.9  2115.1   102.3 2104.62   137.5 2096.54     184 2095.42
   228.5 2090.11   249.2 2083.08   264.2 2083.57   288.3 2069.38   319.3 2069.08
   329.3 2074.03   334.4 2074.39   349.4 2074.05   365.1 2070.42   384.5 2068.44
   444.6 2068.29   474.5 2070.31     523 2073.45   551.6 2071.69     623 2076.11
   734.1 2070.86   839.4 2075.79   894.2 2074.93   936.3 2072.02   952.2 2077.43
   961.6 2084.58   982.6 2112.11   995.3 2123.65  1020.6 2137.73  1049.8 2148.12
#Mann= 3 ,-1,0
       0      .1       0   365.1    .045       0   474.5      .1       0
Bank Sta=365.1,474.5
XS Rating Curve= 0 ,0
Exp/Cntr(USF)=0,0
Exp/Cntr=0.3,0.1

Type RM Length L Ch R = 1 ,6315    ,603.4,603.4,603.4
XS GIS Cut Line= 4
2387262.95972138724454.7718213962387228.67690244724603.617890704
2386867.67651988725274.424184877 2386870.6062472725364.801424726
#Sta/Elev= 30
       0 2116.97   159.1 2106.01   163.6 2103.23   177.2 2089.98   189.7 2087.68
   204.5 2077.27     209 2071.73   213.6 2067.34   231.7 2067.03   299.9 2067.28
   310.8 2071.61     368  2072.2   381.7 2069.56   408.9 2068.29   445.2 2070.13
   464.3 2074.05   490.9 2072.45   517.5 2074.11   585.4 2074.38   645.1 2069.65
   744.7 2072.26   776.8 2075.13   854.1 2070.85   876.8 2073.68   908.6 2073.72
   913.5 2075.19   921.3 2080.41   937.5 2097.56   953.3 2108.73  1004.9 2137.17
#Mann= 3 ,0,0
       0      .1       0     209    .045       0   310.8      .1       0
Bank Sta=209,310.8
XS Rating Curve= 0 ,0
Exp/Cntr=0.3,0.1

Type RM Length L Ch R = 1 ,5712    ,454.4,454.4,454.4
XS GIS Cut Line= 2
2386601.34082376724363.1307907392386702.96317436725381.405016181
#Sta/Elev= 30
       0 2142.55    10.1 2136.91    74.4 2111.12    98.5 2097.64   110.5 2095.71
   125.1 2087.65   154.8 2075.84   166.9 2074.54   178.9 2066.52     191 2063.62
   235.2 2063.53   275.4 2063.81  287.88 2066.61   295.5 2069.81   303.5 2070.12
   379.9 2063.22   412.1 2071.08   464.3 2073.26   746.4 2071.38   765.8 2067.08
   781.9 2070.23   838.2 2068.42   866.3 2071.99   910.5 2073.97   922.6 2077.49
   934.7  2086.5   946.7 2087.58   959.2 2101.47   986.9 2120.68  1023.3 2137.78
#Mann= 3 ,0,0
       0      .1       0   178.9    .045       0  287.88      .1       0
Bank Sta=178.9,287.88
XS Rating Curve= 0 ,0
Exp/Cntr=0.3,0.1

Type RM Length L Ch R = 1 ,5257    ,576.8,576.8,576.8
XS GIS Cut Line= 2
2386152.12976108724390.6819557252386249.17978553725363.787010012
#Sta/Elev= 30
       0 2164.33     6.5 2163.49    54.8 2132.02    66.8 2128.84      95 2112.01
   139.2 2067.34   147.2 2063.94   155.3 2065.23   166.8 2062.39   291.9 2061.69
   319.8 2062.62  330.29 2065.23   360.3 2068.55   404.5 2069.35   470.2 2067.13
   510.4  2062.7   533.1  2063.9   545.2 2062.53   557.9 2067.53   568.9 2069.03
   589.4 2067.42   678.6 2071.01   794.4 2067.47   822.6 2063.13   870.8 2072.89
   886.8  2084.3     911 2097.64   955.2 2111.02   967.3 2118.23   977.9 2119.09
#Mann= 3 ,-1,0
       0      .1       0   155.3    .045       0  330.29      .1       0
Bank Sta=155.3,330.29
XS Rating Curve= 0 ,0
Exp/Cntr=0.3,0.1

Type RM Length L Ch R = 1 ,4680    ,520.4,520.4,520.4
XS GIS Cut Line= 2
2385567.94657447 724572.863191812385744.67249574 725244.74302895
#Sta/Elev= 30
       0 2154.17    25.1 2135.07    37.6 2121.55    58.2 2109.86    78.9 2093.76
   103.7  2068.7     112  2066.2  118.79 2061.21   124.4 2058.01   128.5 2057.53
   186.4 2057.31   219.5 2057.52   235.8 2061.19   252.6 2064.03   273.3 2064.05
     294  2065.8   360.7 2063.37   397.4 2066.35   439.3 2066.26   496.7 2064.66
   504.9 2063.37   517.3  2058.4   521.1 2058.12   554.6 2058.39   571.1 2063.56
   582.7 2069.24   604.2 2084.48   616.6 2090.38   648.8 2096.25   694.7 2099.72
#Mann= 3 ,0,0
       0      .1       0  118.79    .045       0   235.8      .1       0
Bank Sta=118.79,235.8
XS Rating Curve= 0 ,0
Exp/Cntr=0.3,0.1

Type RM Length L Ch R = 1 ,4160    ,604.3,604.3,604.3
XS GIS Cut Line= 2
2385052.41703854724676.7550311232385240.84660382725336.931224251
#Sta/Elev= 30
       0 2194.93    12.9 2181.47    25.4 2171.99    61.6 2133.98    96.1 2108.54
   108.6 2095.15   141.9 2065.96     146 2063.77   166.8 2063.36   171.7 2062.17
   178.1 2058.59   183.5 2056.67   225.1 2056.48   287.5 2056.58   303.7  2058.5
   320.7 2059.39   352.9 2057.66   372.3 2060.15   416.4 2061.45   445.5 2060.76
   462.9 2058.67   509.2 2057.91   528.7 2055.96   541.2 2058.36   557.8 2066.15
   574.5 2067.99   595.3 2075.64   621.5 2082.05     666 2095.74   686.5 2100.39
#Mann= 3 ,0,0
       0      .1       0   178.1    .045       0   303.7      .1       0
Bank Sta=178.1,303.7
XS Rating Curve= 0 ,0
Exp/Cntr=0.3,0.1

Type RM Length L Ch R = 1 ,3556    ,492.6,492.6,492.6
XS GIS Cut Line= 3
2384527.69581764724823.4309428052384508.94237753724946.489934942
2384628.03185577725475.274252801
#Sta/Elev= 30
       0 2147.47      22 2140.17    66.5 2130.92    78.6  2126.6    86.7 2126.69
    90.8 2125.44    98.9 2121.11   115.1 2120.99   147.7 2100.54   188.7 2063.59
     201 2054.68   205.1 2052.22   209.2  2051.8   250.2 2051.85   287.1 2050.35
   296.8 2053.37   307.6 2055.82   315.8 2054.65   344.5 2055.55   400.5 2054.76
   455.3 2057.19   520.9 2054.72   533.2 2053.05   553.7 2053.66   570.1 2059.54
   586.5 2061.13   590.6 2063.29   598.8 2070.22   635.7 2094.52   666.5 2118.42
#Mann= 3 ,-1,0
       0      .1       0     201    .045       0   296.8      .1       0
Bank Sta=201,296.8
XS Rating Curve= 0 ,0
Exp/Cntr=0.3,0.1

Type RM Length L Ch R = 1 ,3063    ,411.7,411.7,411.7
XS GIS Cut Line= 4
2384070.12629588724854.3352445062384026.58680653 725028.02789357
2384116.31474395725472.7663659952384117.73840198725541.101271866
#Sta/Elev= 30
       0 2128.99    44.2 2119.37    93.7 2106.57   118.4 2094.66   139.1 2082.83
   155.5 2075.16   167.9 2067.48     172 2066.19   184.3 2063.05   257.8 2062.04
   266.3 2058.55   274.1 2053.32  275.41 2051.06   278.2 2048.11   285.9 2047.25
   384.3 2047.27   388.4 2047.49   395.3 2051.14   400.6  2054.5   412.8 2054.21
   433.2  2057.2   535.3    2056   548.1 2052.66   567.9 2050.69   588.3 2050.91
   596.5 2052.67   629.1 2054.81   645.2 2063.43   669.2 2079.82   701.1 2104.67
#Mann= 3 ,-1,0
       0      .1       0  275.41    .045       0   395.3      .1       0
Bank Sta=275.41,395.3
XS Rating Curve= 0 ,0
Exp/Cntr=0.3,0.1

Type RM Length L Ch R = 1 ,2651    ,383.7,383.7,383.7
XS GIS Cut Line= 4
2383705.38679867 724831.666755162383654.67100795724977.312102855
2383653.37060306725376.5364041252383641.66695905  725419.4497655
#Sta/Elev= 30
       0 2109.42    24.1 2103.52    35.5 2102.35    80.7 2089.91    94.8 2085.13
   145.6 2064.02   166.1 2058.49   182.1 2059.51   222.1 2059.35   282.1 2061.94
   326.1 2060.53   338.1    2059   346.1  2051.9   350.1 2050.26   371.9 2048.24
   386.1 2045.15   466.1 2045.07   474.1 2045.11   482.1 2048.33   522.1 2051.41
   526.1 2052.44   534.1 2056.72   538.1  2057.9   558.3 2059.54   562.4 2063.75
   566.6 2073.82   574.8 2087.28     579 2093.09   583.1 2097.51   597.9 2110.15
#Mann= 3 ,-1,0
       0      .1       0   371.9    .045       0   482.1      .1       0
Bank Sta=371.9,482.1
XS Rating Curve= 0 ,0
Exp/Cntr(USF)=0,0
Exp/Cntr=0.3,0.1

Type RM Length L Ch R = 1 ,2268    ,257.9,257.9,257.9
XS GIS Cut Line= 2
2383463.88142395724769.7797608792383243.73065769725243.453317859
#Sta/Elev= 30
       0 2102.36    12.6 2098.28    52.3 2087.53   122.8 2061.27   136.1 2058.38
   141.7 2055.95   149.3 2054.24   158.1 2053.32     189 2052.59   211.1 2054.17
   297.4  2055.1   312.5 2056.06   330.2 2050.36   350.5 2049.11   356.6  2047.5
     361 2044.42   365.4 2044.28     457 2044.38   458.1 2044.53  462.03 2049.15
   466.9 2053.38   471.3 2054.76   488.9 2055.87   493.4  2057.8   497.8 2064.09
   502.2  2072.2   505.2 2079.09     511 2090.61   515.4 2097.41   522.3 2104.42
#Mann= 3 ,-1,0
       0      .1       0   350.5    .045       0  462.03      .1       0
Bank Sta=350.5,462.03
XS Rating Curve= 0 ,0
Exp/Cntr(USF)=0,0
Exp/Cntr=0.3,0.1

Type RM Length L Ch R = 1 ,2010    ,760.3,760.3,760.3
XS GIS Cut Line= 3
2383213.76798697724737.0739186342382991.41767099725156.898772007
2383026.13567098725226.942998766
#Sta/Elev= 30
       0 2091.48    20.5 2085.17    77.1 2071.35    86.1 2067.51    99.7 2067.06
   117.8 2060.58   128.5 2054.53   149.5 2048.31     154 2047.75   167.6 2050.59
   193.6 2047.22   208.3 2046.44   232.1 2048.43   262.6 2048.75   267.2 2047.89
   271.7 2044.64   276.2    2044   407.5 2044.01     412  2046.1  415.32 2048.64
   425.6 2051.46   430.1 2051.48   439.2 2049.72   448.2 2050.57   452.8 2053.45
   466.3 2069.66   479.8 2075.42     529 2085.04   542.3 2089.77   553.2 2091.17
#Mann= 3 ,-1,0
       0      .1       0   262.6    .045       0  415.32      .1       0
Bank Sta=262.6,415.32
XS Rating Curve= 0 ,0
Exp/Cntr(USF)=0,0
Exp/Cntr=0.3,0.1

Type RM Length L Ch R = 1 ,1249    ,634.2,634.2,634.2
XS GIS Cut Line= 4
2382262.70028503724745.6709075612382348.97585569724852.468462063
2382399.78028898 725033.229513132382903.77248936725194.073253209
#Sta/Elev= 30
       0 2090.91    66.2 2075.58    91.9 2071.44   112.5 2069.61   142.2 2063.54
   154.7 2059.84     163  2050.7  166.18 2044.44   167.1 2042.95   171.3  2040.5
   237.7 2040.44   266.8 2044.55   292.9 2044.79   308.4 2042.91     325 2048.24
   338.1 2049.09   350.7 2044.73   363.5 2043.27   380.1 2046.63     401 2047.43
   548.1 2047.73     632 2050.17   723.2 2049.57   745.3 2046.83   770.9 2046.36
   786.9 2049.93   804.1 2057.48   820.9 2069.36   824.8 2071.13   854.1 2075.78
#Mann= 3 ,-1,0
       0      .1       0  166.18    .045       0   266.8      .1       0
Bank Sta=166.18,266.8
XS Rating Curve= 0 ,0
Exp/Cntr=0.3,0.1

Type RM Length L Ch R = 1 ,615     ,294.2,294.2,294.2
XS GIS Cut Line= 3
2382190.91084951725601.8922397652382446.39181784725235.775332184
2382905.94874853 725217.29612261
#Sta/Elev= 30
       0 2214.61    30.1 2195.48    44.1 2184.88    54.5 2179.38    93.5 2148.08
   113.5 2133.93   132.6 2118.71   142.2 2108.02   162.3 2072.32   176.5 2056.71
     196 2053.58  215.882041.044   220.4  2038.1   328.9 2037.88   393.6 2037.94
  401.922041.043   410.6 2043.45   423.7 2045.14   496.3 2047.55   556.3  2048.5
   648.4 2047.36   696.4 2048.41   752.5 2047.02   780.5 2048.35   792.5  2050.6
   808.5 2057.13   820.1 2060.36   828.5 2065.47   836.5 2067.73906.3722 2076.66
#Mann= 3 ,-1,0
       0      .1       0  215.88    .045       0  401.92      .1       0
Bank Sta=215.88,401.92
XS Rating Curve= 0 ,0
Exp/Cntr(USF)=0,0
Exp/Cntr=0.3,0.1
